HEC-RAS study SHVRSFK.prj: SHVRSFK

--- SHVRSFK.g01 (geometry) --- (continued)

Type RM Length L Ch R = 1 ,39566   ,393.8,382.8,371
XS GIS Cut Line= 2
2266318.33644353528604.6149994572266711.41407037528502.853786417
#Sta/Elev= 30
       0 3888.03    10.2 3886.49    30.8 3885.09      68 3880.17    79.8 3879.73
    89.7 3878.31   105.2 3878.48   122.5 3873.61   146.5  3875.5   158.9 3875.16
     163 3874.45     1743869.886   176.2 3869.53   202.23869.885   208.5 3870.67
   220.9 3870.53   229.2 3873.03   258.1 3873.24   270.5 3872.49   278.7 3871.06
   311.8 3883.07   324.2 3891.58   328.3  3892.6   340.7 3892.69   344.8 3893.65
   362.1 3904.58   369.6 3908.21   377.9 3909.62   390.3 3913.65     406 3915.22
#Mann= 3 ,-1,0
       0      .1       0     174    .045       0   202.2      .1       0
#XS Ineff= 2 , 0
          127.37 3880.04
Permanent Ineff=
       F       F
Bank Sta=174,202.2
XS Rating Curve= 0 ,0
Exp/Cntr(USF)=0,0
Exp/Cntr=0.3,0.1

Type RM Length L Ch R = 1 ,39183   ,227.4,245,266.6
XS GIS Cut Line= 3
2266358.24280159528919.8752280892266631.60135426528933.842453408
2266829.13782663528762.245113773
#Sta/Elev= 30
       0 3898.83      18 3892.87      38 3888.07      58 3881.84    94.1 3880.36
   130.1 3877.68   150.1 3877.11   154.1 3876.48   170.2 3870.82   174.2 3870.23
   206.2 3870.08   254.3 3871.91   285.1 3871.39   295.7 3870.47   311.5  3871.5
   322.2 3870.59   331.3 3867.78   341.8 3867.06   362.5 3867.62   369.8 3869.33
   407.9 3870.84   424.9 3878.58   433.4 3883.52   438.7 3885.53   445.5 3886.23
   458.9 3885.91   467.4 3889.19     497 3896.17   524.1 3904.37   535.4 3906.52
#Mann= 3 ,-1,0
       0      .1       0   331.3    .045       0   362.5      .1       0
Bank Sta=331.3,362.5
XS Rating Curve= 0 ,0
Exp/Cntr(USF)=0,0
Exp/Cntr=0.3,0.1

Type RM Length L Ch R = 1 ,38938   ,324.2,326.3,320
XS GIS Cut Line= 3
 2266364.2287553 529037.598984352266863.05823098 529103.44447514
2266964.81944402529069.524070794
#Sta/Elev= 30
       0 3893.93    20.1 3889.32    28.2 3889.54     117 3880.64   141.2 3876.73
   177.8 3868.91   193.6 3868.39   262.2 3869.97   274.3 3869.55   282.4 3867.05
   363.1 3869.47   379.2 3867.14   403.4 3868.43   409.5 3867.76   415.5 3866.25
   434.23867.687   443.8 3868.96   463.9 3868.16     472 3868.79     476 3870.23
   492.2 3879.57   503.2  3880.2   512.8 3879.42   529.6 3887.21   542.3 3891.45
   567.6 3893.66     576 3895.19   594.4 3893.88   600.7 3895.42   610.4 3899.32
#Mann= 3 ,-1,0
       0      .1       0   409.5    .045       0   434.2      .1       0
Bank Sta=409.5,434.2
XS Rating Curve= 0 ,0
Exp/Cntr(USF)=0,0
Exp/Cntr=0.3,0.1

Type RM Length L Ch R = 1 ,38612   ,264.7,263,261.4
XS GIS Cut Line= 3
2266386.17725223529257.0839536512266839.11441615529348.868577177
 2266952.8475366529342.882623469
#Sta/Elev= 30
       0 3893.36     6.1 3892.12    18.4 3891.73    91.8  3878.2   113.8 3874.54
   120.6 3874.22   132.6 3870.14     149 3867.43   173.5 3865.54   193.9 3866.79
   210.2 3865.98   246.1 3867.39   263.2 3866.21   276.7 3863.51   295.9 3863.18
     3063863.476   312.2 3864.42   320.4 3867.05   341.1 3868.38   357.1 3867.61
     402 3867.76   442.6 3869.93   463.2 3875.57   491.2 3876.09   504.7  3883.2
   519.9 3889.62   543.3 3891.55   551.3 3890.82   559.3 3888.04     576 3889.51
#Mann= 3 ,-1,0
       0      .1       0   276.7    .045       0     306      .1       0
#XS Ineff= 2 , 0
                          344.89         3869.94
Permanent Ineff=
       F       F
Bank Sta=276.7,306
XS Rating Curve= 0 ,0
Exp/Cntr(USF)=0,0
Exp/Cntr=0.3,0.1

Type RM Length L Ch R = 1 ,38349   ,336.8,326.2,312
XS GIS Cut Line= 3
2266360.23811949529534.4331421312266779.25487907 529592.29736131
2266942.87094709529588.306725505
#Sta/Elev= 30
       0 3904.23    36.3 3897.58    72.6 3888.75    94.6  3881.6     109 3873.63
   141.3 3867.95   165.5 3865.97   213.9 3865.72     218 3865.37   226.3 3862.49
   238.2 3861.69   256.53862.471   270.5 3863.15   278.6 3864.61   302.8 3863.74
     331 3865.28   360.7 3864.69   383.5 3863.05   415.8 3867.01   427.9 3866.31
   439.9 3866.91   471.9    3865   479.9 3865.32   495.9 3869.58   503.9 3870.03
   515.9 3869.68   527.9 3866.95   543.9 3866.97     560 3870.85   586.7 3879.85
#Mann= 3 ,-1,0
       0      .1       0   226.3    .045       0   256.5      .1       0
#XS Ineff= 2 , 0
                          411.27         3870.42
Permanent Ineff=
       F       F
Bank Sta=226.3,256.5
XS Rating Curve= 0 ,0
Exp/Cntr(USF)=0,0
Exp/Cntr=0.3,0.1

Type RM Length L Ch R = 1 ,38022   ,371.9,373.9,374.5
XS GIS Cut Line= 3
2266479.95719366529929.5060868722266869.04418469529793.824469486
2266958.83349031529789.833833681
#Sta/Elev= 30
       0 3905.16    42.6 3892.13    49.6 3887.95    59.5  3880.2    71.4 3875.72
    82.1 3870.65    93.4 3863.99   100.9 3861.69   118.8 3860.91   144.3 3862.67
   169.7 3862.22   182.4 3863.12   207.7 3862.57   217.2 3863.04   224.8 3862.12
   233.2  3862.2   240.5 3860.55   254.4 3859.94   268.2 3860.61   275.6    3863
   280.4 3863.38   326.4 3861.67   364.5 3864.16     390  3863.5   406.9 3867.44
   427.2 3867.37   447.2 3871.09   483.3 3873.81   491.3 3875.12   501.9 3874.27
#Mann= 3 ,-1,0
       0      .1       0   240.5    .045       0   268.2      .1       0
#XS Ineff= 2 , 0
                          363.26         3867.49
Permanent Ineff=
       F       F
Bank Sta=240.5,268.2
XS Rating Curve= 0 ,0
Exp/Cntr(USF)=0,0
Exp/Cntr=0.3,0.1

Type RM Length L Ch R = 1 ,37648   ,252.6,251.9,246.1
XS GIS Cut Line= 2
 2266583.7137246530252.7475871152267006.72111998530143.005102465
#Sta/Elev= 30
       0  3891.5      17 3886.69    37.7  3883.3    62.4 3876.67    70.7 3872.39
    83.1 3863.95    98.5 3858.51   103.8 3857.45   114.9 3859.68     124 3859.08
   128.6 3857.69     141 3857.62   161.6  3860.3   187.1 3859.82   198.8 3857.75
   215.4 3859.19     227 3857.69   240.2  3857.2   248.4 3857.56   262.5 3860.67
   285.5 3862.59     298 3862.34   306.3 3861.26   326.9 3863.16   364.1 3861.25
   376.5 3861.84   409.6 3871.19   417.9 3872.89   426.1 3873.19     437 3871.98
#Mann= 3 ,-1,0
       0      .1       0     227    .045       0   248.4      .1       0
#XS Ineff= 2 , 0
                          289.49         3863.94
Permanent Ineff=
       F       F
Bank Sta=227,248.4
XS Rating Curve= 0 ,0
Exp/Cntr(USF)=0,0
Exp/Cntr=0.3,0.1

Type RM Length L Ch R = 1 ,37397   ,248,236.2,224.8
XS GIS Cut Line= 2
2266635.59199007530496.1763712492267064.58533916530312.607124197
#Sta/Elev= 30
       0 3887.45    31.1 3878.21    70.2 3871.37    74.6 3869.62    87.7 3860.94
      92 3859.36   105.1 3857.82   122.5 3859.21   131.2 3858.43   139.8 3856.59
   155.1 3855.87   164.2 3856.54   174.7 3858.65   188.6 3858.84   218.2 3856.28
   226.9 3858.84   231.3 3859.25   257.3 3857.69     266 3859.18   307.4 3859.18
     333 3855.71   340.9 3855.12     3553855.814   366.1 3860.45   380.6 3860.57
   396.6 3865.15     408 3866.51     427 3867.11   456.7 3873.22   466.6 3872.92
#Mann= 3 ,-1,0
       0      .1       0     333    .045       0     355      .1       0
Bank Sta=333,355
XS Rating Curve= 0 ,0
Exp/Cntr(USF)=0,0
Exp/Cntr=0.3,0.1

Type RM Length L Ch R = 1 ,37160   ,335.3,357.8,379.7
XS GIS Cut Line= 2
2266863.05823098530813.4319177842267158.36528059530462.255966902
#Sta/Elev= 30
       0 3866.69      16 3864.34    26.5 3862.07    43.6 3859.82    54.9 3855.86
    68.3 3854.35   100.3 3854.62   132.3 3855.64   142.9 3855.11   154.3 3855.35
   168.5 3854.48     178 3855.78   194.4 3855.03     213 3856.65   244.1  3856.3
     293 3857.56   307.6 3855.52   312.5  3854.2   318.7 3853.05   334.8 3852.76
     340 3852.97   345.3 3854.18   355.7 3856.45   361.5 3859.37   364.4 3860.13
   393.3 3861.14   406.9    3866   429.7 3868.46     455 3873.27   458.8 3873.38
#Mann= 3 ,-1,0
       0      .1       0   312.5    .045       0   345.3      .1       0
Bank Sta=312.5,345.3
XS Rating Curve= 0 ,0
Exp/Cntr(USF)=0,0
Exp/Cntr=0.3,0.1

Type RM Length L Ch R = 1 ,36803   ,309.5,312.2,314.8
XS GIS Cut Line= 3
2266842.94213963530929.5972790672267129.43156743530835.764920081
2267367.87366037530841.366368422
#Sta/Elev= 30
       0 3875.92      27 3869.86    77.1 3863.56    85.5 3861.06    98.1 3854.83
   106.5 3853.45   127.6 3853.87   161.2 3852.86   170.3 3853.64   203.3 3853.38
   220.2 3854.41   241.2 3853.27   296.2 3854.98   308.2 3854.36315.6801 3852.48
   332.2 3850.98341.27943852.272   348.2  3853.6   380.2  3854.4   396.2 3853.79
   408.2 3854.61   440.2 3854.51   468.3 3852.12   472.3 3853.98   480.3    3860
   496.3 3860.64   500.3 3862.03   512.7 3869.36   528.3 3871.91     540 3871.72
#Mann= 3 ,-1,0
       0      .1       0315.6801    .045       0341.2794      .1       0
Bank Sta=315.6801,341.2794
XS Rating Curve= 0 ,0
Exp/Cntr(USF)=0,0
Exp/Cntr=0.3,0.1

Type RM Length L Ch R = 1 ,36490   ,154.8,143.9,128
XS GIS Cut Line= 2
2266871.03950259531046.8841124042267323.97666651531128.692146416
#Sta/Elev= 30
       0 3886.48    25.5 3880.32    45.9 3876.18    62.1 3871.29    70.3  3867.5
    86.5 3854.76      89 3853.46    94.6 3851.66   106.2 3849.77   110.9 3849.48
   132.5 3849.83   147.4 3851.59   167.8 3851.21   171.9 3850.52     180 3852.28
   192.2  3852.6   220.6 3852.15   232.8 3851.21     244  3852.7   285.3  3852.7
   297.9 3850.65   301.9 3850.55   312.8 3852.85   330.4 3851.94   354.8 3852.38
     367  3854.5   407.6 3855.74   415.8 3857.73   452.3 3870.61   460.3 3872.04
#Mann= 3 ,-1,0
       0      .1       0   106.2    .045       0   132.5      .1       0
Bank Sta=106.2,132.5
XS Rating Curve= 0 ,0
Exp/Cntr(USF)=0,0
Exp/Cntr=0.3,0.1

Type RM Length L Ch R = 1 ,36347   ,166,152.7,135.1
BEGIN DESCRIPTION:
Structure XS 4
END DESCRIPTION:
XS GIS Cut Line= 3
2266885.00672791531258.3878100932267180.31377752531138.668735929
2267335.94857393531164.607868665
#Sta/Elev= 30
       0  3907.5    24.9 3899.46    37.9 3893.51    64.8 3885.46    72.5 3884.17
    81.1 3881.07   102.7 3870.37   110.9 3864.65   123.1 3851.45   128.6 3848.81
   145.9 3848.18   158.8 3848.65   163.1 3851.17   167.4 3852.04   214.9 3851.47
   223.5 3850.52   236.5 3851.59   262.4 3851.16     289 3852.24   298.2 3851.75
   305.6 3850.08   314.2 3851.37   330.7 3851.27   342.8 3852.68   359.1 3853.09
   367.2 3854.46   403.7 3855.39   452.3 3871.48   466.7 3873.07   476.4 3871.82
#Mann= 3 ,-1,0
       0      .1       0   128.6    .045       0   158.8      .1       0
Bank Sta=128.6,158.8
XS Rating Curve= 0 ,0
Exp/Cntr(USF)=0,0
Exp/Cntr=0.5,0.3

Type RM Length L Ch R = 1 ,36194   ,71.1,70.9,68.3
BEGIN DESCRIPTION:
Structure XS 3
END DESCRIPTION:
XS GIS Cut Line= 3
2267004.72580208531457.9196003672267176.32314171531202.518908817
2267302.02816958531224.467405747
#Sta/Elev= 30
       0 3864.07       3  3864.2    13.4 3862.96      29 3863.48    57.8  3861.4
    85.1 3861.73   106.8 3856.86   111.7  3854.4   118.3 3850.05   126.2 3847.12
   140.6 3846.66   158.7 3847.09   171.2 3847.71     176 3848.75     184 3848.19
   193.3 3848.89     207  3848.7   246.7 3850.44   271.6 3853.49   278.7 3852.94
   285.9 3851.47   299.9 3851.94   323.8 3851.53   331.9 3854.11     336 3854.78
   368.5 3854.19   380.6 3854.62   388.8  3856.8   425.3 3869.47   435.3 3871.43
#Mann= 3 ,-1,0
       0      .1       0   126.2    .045       0   158.7      .1       0
#XS Ineff= 2 , 0
            96.5  3858.5   193.5            3858
Permanent Ineff=
       F       F
Bank Sta=126.2,158.7
XS Rating Curve= 0 ,0
Exp/Cntr(USF)=0,0
Exp/Cntr=0.5,0.3

Type RM Length L Ch R = 1 ,36123   ,113.9,139.1,179.4
BEGIN DESCRIPTION:
Structure XS 2
END DESCRIPTION:
XS GIS Cut Line= 3
2267034.65557062531515.7838195462267226.20608928531252.401856385
2267290.05626217531262.378445899
#Sta/Elev= 30
       0 3857.29    16.2 3857.39    29.8 3856.96    40.2 3855.39    47.7  3855.2
    52.7 3854.77    71.7 3851.73    87.3  3850.2    91.7 3849.99   103.2 3850.19
   111.8 3849.86   118.2 3848.87     125  3847.2   136.8 3846.92   166.4 3847.21
   171.4 3848.03   174.8 3849.17   181.3 3850.44   191.9 3851.08   217.7 3851.49
   233.8 3851.26   249.2 3852.66   260.7 3853.07     295 3853.56   314.8 3853.56
   338.6 3854.15   343.9 3855.35   368.1 3863.82   384.1    3869   390.3 3870.21
#Mann= 3 ,-1,0
       0      .1       0     125    .045       0   166.4      .1       0
#XS Ineff= 2 , 0
           122.8  3858.5   171.2            3858
Permanent Ineff=
       F       F
Bank Sta=125,166.4
XS Rating Curve= 0 ,0
Exp/Cntr(USF)=0,0
Exp/Cntr=0.5,0.3

Type RM Length L Ch R = 1 ,35984   ,88.7,88.3,87.6
BEGIN DESCRIPTION:
Structure XS 1
END DESCRIPTION:
XS GIS Cut Line= 2
2267034.65557062531519.774455351 2267244.1639504531571.652720823
#Sta/Elev= 30
       0  3856.9     5.7 3856.53     9.8 3855.93    13.9  3854.4      18 3852.29
    22.1 3851.03    34.5 3848.91    38.7 3848.53    55.3 3848.82    63.4 3848.47
    67.5 3848.88    75.7 3848.96    79.9 3848.59      84  3847.4    86.93846.899
    96.3 3846.54   104.8 3846.56   112.8 3847.05   116.9 3849.82   121.1 3852.03
   133.4  3852.1   145.8 3853.15     154 3855.12   166.4 3858.68   174.6 3860.58
   180.8  3861.6   188.9 3863.38   203.5 3865.06   207.6 3865.77   215.8 3865.73
#Mann= 3 ,-1,0
       0      .1       0    86.9    .045       0   112.8      .1       0
Bank Sta=86.9,112.8
XS Rating Curve= 0 ,0
Exp/Cntr(USF)=0,0
Exp/Cntr=0.3,0.1

Type RM Length L Ch R = 1 ,35895   ,167.1,155.8,149.4
BEGIN DESCRIPTION:
Structure XS 4
END DESCRIPTION:
XS GIS Cut Line= 2
2266881.01609211531577.6386745312267254.14053992531661.442026446
#Sta/Elev= 30
       0 3885.61    12.3 3879.91    15.7 3879.19    27.8 3879.21    35.7 3877.61
    39.1 3876.19    44.2 3872.67    52.4 3864.93    64.7 3858.06    89.3 3855.84
    93.4 3854.66    97.5 3852.44   101.6 3851.19   146.7 3850.97     163 3851.45
   171.3 3849.73   183.6 3848.33     200 3848.37   212.3 3846.73   219.9  3846.7
   236.6 3846.28   253.3 3846.75   253.3 3846.77   257.4 3850.51   261.5 3852.07
   283.5 3852.89   351.7 3861.81     364 3862.65   376.3 3864.76   382.4 3864.65
#Mann= 3 ,-1,0
       0      .1       0   219.9    .045       0   253.3      .1       0
Bank Sta=219.9,253.3
XS Rating Curve= 0 ,0
Exp/Cntr(USF)=0,0
Exp/Cntr=0.5,0.3

Type RM Length L Ch R = 1 ,35740   ,120.4,121.2,121
BEGIN DESCRIPTION:
Structure XS 3
END DESCRIPTION:
XS GIS Cut Line= 4
2266714.35235594531755.3246133582266921.86541782531819.174786246
2267003.67345183531779.2684281912267310.95240885 531771.28715658
#Sta/Elev= 30
       0 3919.97    22.1 3911.06    38.1 3900.49    64.7 3900.71   127.5 3861.41
   148.4  3860.6   156.8 3854.44   165.1 3851.51     186 3851.42     207 3854.26
   223.3 3855.09   250.2 3851.61   308.6 3848.47   332.6 3848.35   341.9 3845.49
   344.7 3844.33   351.7 3844.18   388.6 3845.56     401 3850.81   428.7 3853.84
   452.7 3854.28   460.7 3856.23   468.7 3860.24   496.7 3862.82   521.3 3863.35
   552.7 3866.68   576.7 3860.79   583.7  3860.9   600.7 3863.86   615.5 3862.43
#Mann= 3 ,-1,0
       0      .1       0   341.9    .045       0   388.6      .1       0
#XS Ineff= 2 , 0
             317  3866.5     423            3866
Permanent Ineff=
       F       F
Bank Sta=341.9,388.6
XS Rating Curve= 0 ,0
Exp/Cntr(USF)=0,0
Exp/Cntr=0.5,0.3

Type RM Length L Ch R = 1 ,35619   ,180.7,188.2,196.8
BEGIN DESCRIPTION:
Structure XS 2
END DESCRIPTION:
XS GIS Cut Line= 4
2266735.35788521531874.9410420382266942.87094709531938.791214926
 2267024.6789811531898.8848568712267331.95793812 531890.90358526
#Sta/Elev= 30
       0 3884.21    13.4 3874.77    21.8 3870.93    50.4 3866.78    63.6 3862.91
    98.5 3862.03   114.5 3866.79   149.7 3867.39   172.1 3863.88   193.4 3851.52
   217.1 3845.65   240.8 3845.31   315.6 3847.73   326.4 3844.31   335.6 3843.96
   356.63844.412   359.6 3845.03   367.7  3851.1   371.6 3851.71   415.7 3853.17
   427.7 3860.42   439.7 3863.89   459.7  3864.4   471.7 3861.46   475.7 3861.37
   503.7 3861.76   512.1 3863.13   527.7 3862.19   583.7 3861.93   615.5 3862.77
#Mann= 6 ,-1,0
       0      .1       0  257.11     .08       0  307.11     .07       0
   326.4    .045       0   356.6     .07       0  368.14      .1       0
#XS Ineff= 2 , 0
             305  3866.5     385            3866
Permanent Ineff=
       F       F
Bank Sta=326.4,356.6
XS Rating Curve= 0 ,0
Exp/Cntr(USF)=0,0
Exp/Cntr=0.5,0.3

Type RM Length L Ch R = 1 ,35430   ,164.3,164.9,164.5
BEGIN DESCRIPTION:
Structure XS 1
END DESCRIPTION:
XS GIS Cut Line= 2
2266711.41407037531986.6788445912267248.15458621532152.290230518
#Sta/Elev= 30
       0 3882.76    13.4 3873.45    21.7 3870.32      41  3865.9    55.2 3865.82
    63.6 3868.24    84.5 3868.89   101.8 3866.61   108.2 3864.23   130.6 3849.68
   147.3 3845.05   159.4  3844.5   189.2 3845.28   198.4 3844.36   239.4 3845.87
   256.1 3844.87   302.2 3845.93   309.7  3843.7   331.5 3843.41   338.5  3843.7
   348.1 3846.61   356.6 3850.51   385.9 3850.47   390.1  3851.3   405.7 3856.16
   415.2 3857.49   436.1 3866.14   452.9 3870.01   466.5 3871.28   561.7 3873.34
#Mann= 6 ,-1,0
       0      .1       0     180     .07       0     280     .08       0
   309.7    .045       0   338.5     .08       0     390      .1       0
Bank Sta=309.7,338.5
XS Rating Curve= 0 ,0
Exp/Cntr(USF)=0,0
Exp/Cntr=0.3,0.1

Type RM Length L Ch R = 1 ,35266   ,184,183.7,181.5
XS GIS Cut Line= 3
2266661.53112281532128.3464156852267042.63684223532258.042079363
2267250.14990411532164.262137935
#Sta/Elev= 30
       0 3886.38       7 3884.21    19.7 3875.36    23.9 3873.25    40.8 3869.04
    78.8 3870.98    87.3 3869.97    91.5 3868.17     100 3858.53   101.9 3857.22
   119.4 3851.24     138 3847.86   167.6  3845.7   201.2 3844.69   258.1 3845.58
   270.7 3842.79   286.5  3842.2   303.9 3842.66   315.5 3844.27   332.4  3844.2
     345 3848.13   357.7  3849.5   426.2 3849.56   448.2 3850.48   487.7 3854.89
   505.2 3858.68   534.4 3867.47   550.4 3869.99   579.8 3872.19   630.3 3873.27
#Mann= 5 ,-1,0
       0      .1       0     230     .08       0   270.7    .045       0
   303.9     .08       0     340      .1       0
Bank Sta=270.7,303.9
XS Rating Curve= 0 ,0
Exp/Cntr(USF)=0,0
Exp/Cntr=0.3,0.1

Type RM Length L Ch R = 1 ,35082   ,162.7,155.9,156.3
XS GIS Cut Line= 2
2266677.49366603532321.8922522512267254.14053992 532511.44745301
#Sta/Elev= 30
       0  3873.7    11.2  3874.6    28.1 3874.75    32.3 3874.32    40.7 3871.56
    44.9 3871.04    57.6 3871.12      66 3870.43    71.3 3868.37    78.6 3863.31
    82.8 3861.15    95.5    3857   112.3 3849.39   124.9 3846.05   133.4  3845.5
     146 3842.59   158.6 3842.29     167 3843.89   174.7 3844.09   217.6 3843.19
   234.4 3842.43   241.1 3841.44   263.9 3841.13   268.53841.577   276.5 3847.25
   415.5 3846.91   474.4 3847.43   543.4 3849.28   568.8 3851.61     607 3851.95
#Mann= 6 ,-1,0
       0      .1       0     220     .08       0   241.1    .045       0
   268.5     .08       0     320      .1       0     550     .08       0
#XS Ineff= 2 , 0
                          278.64         3850.15
Permanent Ineff=
       F       F
Bank Sta=241.1,268.5
XS Rating Curve= 0 ,0
Exp/Cntr(USF)=0,0
Exp/Cntr=0.3,0.1

Type RM Length L Ch R = 1 ,34926   ,222.8,193.5,158.1
XS GIS Cut Line= 3
2266656.28691807532481.4279795582266901.33648898532535.539872189
2267252.29076405532561.822791467
#Sta/Elev= 30
       0 3878.75     8.1 3878.09    16.3  3876.1    28.6 3869.49    36.6 3867.31
    44.9 3868.73    57.2 3869.44    69.5 3868.64    76.9 3867.32    85.9 3861.42
      97 3855.74   120.5 3849.46   143.3 3840.61   167.5 3840.12   173.7  3840.6
   180.1 3842.53     191  3843.9   208.8 3842.76   221.2 3845.69     242 3846.64
   358.1 3845.97   422.3 3847.11   438.7 3846.07   458.4 3846.24   470.4 3847.03
   514.5 3847.16   530.6  3848.5   542.8 3848.35   582.7 3850.73   602.9  3851.2
#Mann= 6 ,-1,0
       0      .1       0   143.3    .045       0   173.7      .1       0
     230     .08       0  330.95     .07       0  430.95     .08       0
#XS Ineff= 2 , 0
                          237.23         3848.16
Permanent Ineff=
       F       F
Bank Sta=143.3,173.7
XS Rating Curve= 0 ,0
Exp/Cntr(USF)=0,0
Exp/Cntr=0.3,0.1

Type RM Length L Ch R = 1 ,34732   ,122.7,150.7,176
BEGIN DESCRIPTION:
Structure - abutments, no deck
END DESCRIPTION:
XS GIS Cut Line= 4
 2266619.9546473532724.9314963992266763.73767629   532737.299929
2266829.59990952532640.1409909452267249.37537134532583.798786959
#Sta/Elev= 30
       0  3863.8    32.3 3863.48    52.4 3859.61    64.5 3852.31      67 3851.82
    92.9  3849.8   108.6 3845.69   124.7  3845.1   140.7 3846.49   156.2  3841.9
   166.5 3841.09   170.6 3839.68   173.5 3838.63   178.3 3838.33   202.1 3838.34
   207.3 3839.69   212.1 3842.66   216.9 3844.52   228.2 3845.68   264.3 3846.27
   289.2 3845.21   304.6 3846.04   409.6 3844.27   445.9 3845.54   466.1 3845.14
   510.5 3846.28   554.9 3845.47   590.4 3846.08   618.9 3848.36   685.2 3850.48
#Mann= 8 ,-1,0
       0      .1       0   170.6    .045       0   207.3      .1       0
  311.69     .08       0  411.69     .07       0  511.69     .08       0
  611.69      .1       0  631.69     .08       0
#XS Ineff= 2 , 0
                          253.31         3848.23
Permanent Ineff=
       F       F
Bank Sta=170.6,207.3
XS Rating Curve= 0 ,0
Exp/Cntr(USF)=0,0
Exp/Cntr=0.5,0.3

Type RM Length L Ch R = 1 ,34582   ,114.6,97.4,83
BEGIN DESCRIPTION:
Structure - abutments, no deck
END DESCRIPTION:
XS GIS Cut Line= 3
2266623.04675545 532843.204633152266912.93189455532837.020416849
2267266.20525072532603.566251497
#Sta/Elev= 30
       0 3851.83    21.1  3851.3    53.1 3848.71   109.5 3847.45   133.2  3847.6
   157.2 3847.04   165.2 3844.04   173.2 3839.29   175.5 3838.67   177.2 3838.15
   181.2 3838.01   201.2 3837.97   209.2 3838.62   229.2 3841.71   237.2  3845.4
   241.2 3845.86   308.2 3844.77     337 3845.44   361.5 3844.19   375.3 3844.35
   393.2 3843.76   418.5 3844.23   448.1 3843.55   500.1 3843.72   509.6 3844.16
   543.2  3844.3   591.1 3845.91   635.7 3846.83   676.1 3848.95   713.4 3850.09
#Mann= 7 ,-1,0
       0      .1       0   175.5    .045       0   209.2      .1       0
     260     .08       0  369.95     .07       0  489.95     .08       0
  609.95      .1       0
#XS Ineff= 2 , 0
                          258.32         3846.83
Permanent Ineff=
       F       F
Bank Sta=175.5,209.2
XS Rating Curve= 0 ,0
Exp/Cntr(USF)=0,0
Exp/Cntr=0.5,0.3

Type RM Length L Ch R = 1 ,34484   ,230.2,230.9,231.4
XS GIS Cut Line= 2
2266631.60135426533070.1364657762267266.11244733532641.143116688
#Sta/Elev= 30
       0 3844.82    12.6 3843.56    24.8 3844.97      49 3845.38    63.5 3843.23
    73.1 3843.31    82.8 3842.18   102.1 3841.63   131.1 3841.67   140.7 3842.35
   155.2 3842.31   176.8 3841.17   203.5 3841.73   211.4 3841.04     220 3837.96
   232.5 3837.31   256.6 3837.93   266.1 3840.05   283.4 3841.16   304.9 3840.27
     329 3842.69   380.2 3844.31   430.4 3844.78   469.1 3843.75   577.3 3843.68
   609.1  3844.1   637.3 3845.44   691.2 3845.52   734.6 3848.05   765.9 3848.67
#Mann= 7 ,-1,0
       0      .1       0     180     .08       0     220    .045       0
   256.6     .08       0     420     .07       0     540     .08       0
     660      .1       0
#XS Ineff= 2 , 0
          193.18 3843.61
Permanent Ineff=
       F       F
Bank Sta=220,256.6
XS Rating Curve= 0 ,0
Exp/Cntr(USF)=0,0
Exp/Cntr=0.3,0.1

Type RM Length L Ch R = 1 ,34253   ,363.5,352.6,345.2
XS GIS Cut Line= 2
2266685.47493764533305.583978298 2267315.9953949532892.553172432
#Sta/Elev= 30
       0 3888.08       8 3887.38    31.9 3879.23    45.6 3871.09      51 3865.31
    71.6 3847.53    79.7 3843.93   170.6 3838.21   218.4  3839.1   234.3 3837.92
     271 3838.19   291.2 3839.33   294.9 3839.12   302.7 3836.39   314.3 3836.01
   331.6 3836.32   343.2 3839.39   354.7 3839.24     381 3842.74     410 3842.33
   428.8 3843.71   433.6  3843.1   444.3  3844.6   467.1 3844.78   528.1 3841.64
   562.7 3843.56   723.4 3843.55     738 3844.84   749.2 3849.07   753.8 3849.38
#Mann= 7 ,-1,0
       0      .1       0     230     .08       0   302.7    .045       0
   331.6     .08       0     410      .1       0     470     .08       0
     710      .1       0
#XS Ineff= 2 , 0
           219.9 3845.59
Permanent Ineff=
       F       F
Bank Sta=302.7,331.6
XS Rating Curve= 0 ,0
Exp/Cntr(USF)=0,0
Exp/Cntr=0.3,0.1

Type RM Length L Ch R = 1 ,33901   ,280.9,280.2,276.9
XS GIS Cut Line= 4
2266954.84285451533636.8067501522267090.24672867533440.923317401
 2267139.7037514533399.5192831852267411.28556419533064.494487383
#Sta/Elev= 30
       0 3932.52    38.1 3919.28      53 3910.14    66.8 3908.76    72.5    3907
    84.1 3899.16    93.8 3894.92   104.2 3889.21   116.3 3885.61     136 3876.28
   145.4 3870.25   170.3 3856.23     179 3848.84   185.2 3842.29   199.1  3837.1
204.87923834.116   208.6  3833.2   220.4 3833.03 236.0763833.997   256.4 3836.38
   268.9 3836.65   292.8 3835.42   309.7  3837.6   322.4 3836.23   377.7 3837.81
   424.1 3837.84   600.4 3842.42   671.8 3842.34   702.1 3848.35   733.9  3849.3
#Mann= 5 ,-1,0
       0      .1       0204.8792    .045       0 236.076      .1       0
  522.63     .08       0  582.63      .1       0
#XS Ineff= 1 ,-1
  403.06   702.6 3842.84
Permanent Ineff=
       F
Bank Sta=204.8792,236.076
XS Rating Curve= 0 ,0
Exp/Cntr(USF)=0,0
Exp/Cntr=0.3,0.1

Type RM Length L Ch R = 1 ,33621   ,295.4,310.8,317.9
XS GIS Cut Line= 4
2267176.32314171533746.5492348032267296.04221587533634.811432249
2267443.69574068533393.3779660192267525.50377469533335.513746839
#Sta/Elev= 30
       0 3895.65    10.7 3889.62    21.7 3885.18    37.2 3874.64      43 3871.96
    60.6 3867.13    85.8 3861.54   103.8 3855.48   142.4 3847.11   163.8  3839.9
   170.9 3836.36   176.7 3835.27   188.3 3835.04   194.1 3832.69   216.6 3832.03
   241.33832.588   248.4  3834.7     264 3834.03   282.9 3834.92   307.6 3834.47
   334.5 3836.33   353.2 3835.84   414.2 3837.51   447.1 3840.84   470.2 3841.23
   486.5 3846.25   491.4 3846.75   506.1 3846.85   516.4 3844.23     547 3845.25
#Mann= 5 ,-1,0
       0      .1       0   194.1    .045       0   241.3      .1       0
  476.77     .08       0  486.77      .1       0
Bank Sta=194.1,241.3
XS Rating Curve= 0 ,0
Exp/Cntr(USF)=0,0
Exp/Cntr=0.3,0.1

Type RM Length L Ch R = 1 ,33310   ,248.5,269.7,282.7
XS GIS Cut Line= 2
2267323.97666651533884.2261700912267697.10111432533654.764611277
#Sta/Elev= 30
       0 3876.96    13.5 3870.99    16.9 3870.04    28.4 3868.42    37.8 3865.54
    47.2 3863.59      78 3858.56    92.5 3854.98   118.7 3850.55   131.7 3846.93
   136.4 3844.85   165.2 3838.73   204.3 3833.07     235 3832.57   261.1  3834.1
   272.6  3832.9   287.3 3833.81   300.8 3830.81   310.2    3830   328.9 3830.12
   332.8 3830.79   341.8 3833.88   348.4 3838.06   366.5 3840.67     392  3840.4
   394.9 3840.98   406.5 3846.65   415.3 3849.38   418.2 3850.06     438 3851.44
#Mann= 3 ,-1,0
       0      .1       0   300.8    .045       0   332.8      .1       0
Bank Sta=300.8,332.8
XS Rating Curve= 0 ,0
Exp/Cntr(USF)=0,0
Exp/Cntr=0.3,0.1

Type RM Length L Ch R = 1 ,33040   ,332.6,317.4,300.6
XS GIS Cut Line= 2
2267359.89238876533952.066978784 2267748.9793798533995.963972644
#Sta/Elev= 30
       0  3877.8    12.4 3872.63    24.4 3869.36    44.6 3865.38    72.7 3857.69
    96.9 3851.75     113 3844.94     117 3842.72   129.1 3839.07   137.1 3835.75
   141.2  3834.6   149.6 3833.76   173.4 3833.07   181.4 3831.62   187.93829.427
     193 3828.31   197.5 3828.23   225.5 3828.52   233.8 3829.56     240 3831.43
   245.8 3834.48   249.9 3835.86   261.9 3837.18   282.1 3838.18   308.7 3838.26
   326.3 3837.25   334.4  3838.8   346.5 3845.24   350.5 3846.31   391.6 3848.09
#Mann= 3 ,-1,0
       0      .1       0   187.9    .045       0   233.8      .1       0
Bank Sta=187.9,233.8
XS Rating Curve= 0 ,0
Exp/Cntr(USF)=0,0
Exp/Cntr=0.3,0.1

Type RM Length L Ch R = 1 ,32723   ,301.2,301.5,303
XS GIS Cut Line= 2
 2267463.6489197534347.1399235262267766.93724092534217.444259848
#Sta/Elev= 30
       0 3862.39     9.3 3857.31    17.1 3854.74      31 3852.31    44.1 3851.64
    52.8  3848.8    70.2 3846.06    91.9 3844.72    96.3 3843.92   105.5 3839.45
     118 3835.42   126.7 3830.91   131.1 3830.11   139.8 3830.15   148.5 3827.99
   157.2 3827.38   183.3  3827.5   185.7 3827.96   187.8 3828.51   190.8 3830.39
   196.3 3834.88     200 3835.72   235.5 3836.55   244.2 3837.27   270.3 3835.85
     279 3837.22   283.3  3838.6   296.4 3845.88   300.7 3847.66   329.9 3850.34
#Mann= 3 ,-1,0
       0      .1       0   148.5    .045       0   185.7      .1       0
Bank Sta=148.5,185.7
XS Rating Curve= 0 ,0
Exp/Cntr(USF)=0,0
Exp/Cntr=0.3,0.1

Type RM Length L Ch R = 1 ,32421   ,319,331.4,350.8
XS GIS Cut Line= 2
2267561.41949694534624.4891120062267842.75932122 534510.75599155
#Sta/Elev= 30
       0 3853.12    16.9 3845.32    29.2 3840.86    32.3 3840.13    54.7  3837.9
      72 3831.64    80.6  3829.7    93.6 3828.41   106.5  3829.2   110.8 3828.59
   115.1 3826.61   119.5 3825.49   145.3 3825.13   152.1 3825.44   162.6 3828.01
   171.2 3828.55   175.6 3829.49   184.2 3833.92   188.5 3834.48   195.1  3834.2
   214.4 3835.13   227.3  3836.8   244.6 3836.52   248.9 3835.67   261.8 3837.02
   270.5 3839.51   274.8 3841.56   283.4 3847.34   287.7 3849.57   303.5 3851.62
#Mann= 3 ,-1,0
       0     .12       0   119.5    .045       0   152.1      .1       0
Bank Sta=119.5,152.1
XS Rating Curve= 0 ,0
Exp/Cntr(USF)=0,0
Exp/Cntr=0.3,0.1

Type RM Length L Ch R = 1 ,32090   ,291.9,295.9,300.2
XS GIS Cut Line= 2
2267587.35862967534865.9225782372267894.63758669534935.758704832
#Sta/Elev= 30
       0 3856.44     4.9 3853.79    13.4 3850.54    17.2 3849.53    25.4 3846.19
    33.9 3841.95    50.1 3837.55    62.4 3835.12    68.8  3832.7    73.6  3831.4
    82.9 3829.41    91.1  3828.3     107 3824.43   115.7 3825.69   123.9 3825.43
   132.1 3824.51   136.2 3823.83   143.8 3823.48   156.7 3823.56   164.9 3824.42
     169  3827.1   173.1  3828.8   185.4 3831.07   193.6 3834.17   205.9 3835.61
     247 3836.59   257.4 3839.53   274.1 3842.22   292.1 3844.57   315.1 3846.52
#Mann= 4 ,-1,0
       0     .12       0      90      .1       0   132.1    .045       0
   164.9      .1       0
Bank Sta=132.1,164.9
XS Rating Curve= 0 ,0
Exp/Cntr(USF)=0,0
Exp/Cntr=0.3,0.1

Type RM Length L Ch R = 1 ,31794   ,186.8,193.3,197.4
XS GIS Cut Line= 2
2267515.52718517  535131.29985932267808.83891688535245.032979756
#Sta/Elev= 30
       0 3845.84     5.2 3844.88    13.6 3844.47    29.8 3841.53    60.8 3838.14
    69.3 3835.83   103.7 3829.25   107.9 3827.71   113.2 3824.73   115.8 3823.67
   119.33822.861   125.1 3822.52   159.4 3822.96   178.2 3827.35   185.2 3828.56
   189.5 3828.54     206 3826.69   219.5 3827.06   223.8  3828.8   228.1 3831.33
   232.4 3833.36   236.7  3834.3   249.5 3835.73   275.3 3836.35   279.6 3836.23
   286.4 3835.19   289.5 3835.08   296.7 3836.09   304.9 3838.05   314.6 3839.69
#Mann= 4 ,-1,0
       0     .12       0      60      .1       0   119.3    .045       0
   159.4      .1       0
Bank Sta=119.3,159.4
XS Rating Curve= 0 ,0
Exp/Cntr(USF)=0,0
Exp/Cntr=0.3,0.1

Type RM Length L Ch R = 1 ,31601   ,224.3,224.4,224.9
XS GIS Cut Line= 2
2267443.69574068535278.9533841032267711.06833964535440.574134224
#Sta/Elev= 30
       0 3849.61      12 3843.61    19.8 3840.79    28.6 3837.01    33.3 3835.88
    42.8 3834.28      52 3833.34    61.3 3831.72    66.2 3831.31   103.4 3829.88
   112.7 3828.33   126.8 3824.95   133.1 3823.84   141.8 3821.65   145.5 3821.24
   173.8 3821.35   182.8 3821.64   189.9 3822.78   206.2 3826.04   210.9 3828.08
   217.5 3831.95   220.8 3833.22   224.9 3834.04   234.3 3834.73     244 3835.98
   262.3 3835.74   271.7 3835.01     281 3835.63     309 3840.69   312.4 3841.07
#Mann= 4 ,-1,0
       0      .1       0     140     .12       0   141.8    .045       0
   182.8      .1       0
Bank Sta=141.8,182.8
XS Rating Curve= 0 ,0
Exp/Cntr(USF)=0,0
Exp/Cntr=0.3,0.1

Type RM Length L Ch R = 1 ,31376   ,184,188.4,192.8
XS GIS Cut Line= 2
2267302.02816958535452.5460416412267611.30244451535644.096560303
#Sta/Elev= 30
       0 3844.36    16.5 3840.38    26.1 3838.47    35.5 3837.47    40.2 3836.61
    54.1 3830.99      62  3828.3    73.1 3826.49    77.8 3825.96   101.3 3824.95
   141.5 3824.23   173.4 3825.19   176.6 3824.85     188 3822.24   191.1 3821.84
   222.8 3821.05   227.2 3822.24   233.1 3825.18   242.5 3831.34   247.2 3832.95
   266.4 3835.18   275.4 3834.46   284.8 3834.45   292.6 3833.78   308.4 3833.76
   312.7 3834.56   317.8 3836.14   322.5  3837.1   339.1 3837.74   363.8 3840.35
#Mann= 3 ,-1,0
       0     .12       0     188    .045       0   227.2      .1       0
Bank Sta=188,227.2
XS Rating Curve= 0 ,0
Exp/Cntr(USF)=0,0
Exp/Cntr=0.3,0.1

Type RM Length L Ch R = 1 ,31188   ,330.3,321.3,315.3
XS GIS Cut Line= 2
2267198.27163864535570.2697979022267473.62550922535799.731356716
#Sta/Elev= 30
       0 3844.59    18.1 3840.92    34.7  3836.9    44.1 3834.96    57.4 3831.07
    68.7 3826.74    71.6 3825.99    80.6 3824.49     100 3824.05   127.4 3823.98
   151.1 3824.84   160.7 3825.55   165.3 3825.52   174.3 3824.79     188 3822.99
   213.6 3820.97   247.2 3820.29   252.4 3820.33   256.2 3820.83   261.9 3822.79
   270.4 3827.21   278.4 3830.76   283.6 3832.34   287.4 3832.89   307.3 3833.74
   324.3 3833.42   335.7 3832.34   351.3 3832.16   354.4 3832.29   358.4 3833.02
#Mann= 5 ,-1,0
       0     .12       0     100      .1       0   213.6    .045       0
   256.2     .12       0     270      .1       0
Bank Sta=213.6,256.2
XS Rating Curve= 0 ,0
Exp/Cntr(USF)=0,0
Exp/Cntr=0.3,0.1

Type RM Length L Ch R = 1 ,30867   ,368,360,353.8
XS GIS Cut Line= 2
2267038.64620642535901.4925697562267361.88770666536047.150776655
#Sta/Elev= 30
       0 3859.36      13 3857.33    22.1 3855.45    46.3 3849.75    58.7 3846.52
    63.1 3845.11    86.9 3833.08   109.8 3820.91   112.8  3819.6   114.93818.955
   115.8 3818.66   120.1 3818.44   127.9 3818.33   146.5 3818.37   152.1 3818.81
   168.4 3822.15   179.4  3823.4   190.3  3823.9   203.5 3825.19   216.7 3824.95
     243 3825.66   282.5 3827.14   291.3 3827.13   295.6 3827.68   308.8 3830.65
   313.2 3830.99   320.5 3830.81   326.3 3831.06     340 3830.81   354.5 3830.95
#Mann= 5 ,-1,0
       0      .1       0      50     .12       0   114.9    .045       0
   152.1     .12       0     260      .1       0
Bank Sta=114.9,152.1
XS Rating Curve= 0 ,0
Exp/Cntr(USF)=0,0
Exp/Cntr=0.3,0.1

Type RM Length L Ch R = 1 ,30507   ,395.9,396.1,397.5
XS GIS Cut Line= 4
2266938.49156044 536211.986357922267023.59959204 536296.94914574
2267173.09713782536324.9799355742267288.44969511536309.658898925
#Sta/Elev= 30
       0 3847.54       8 3846.02      25 3843.95    53.2 3837.74    61.4 3836.29
    92.3  3830.2   112.3 3824.36   124.9 3822.56   133.1 3820.78   141.2 3819.97
151.92053818.311   157.5  3817.7   161.5 3817.65   198.2 3818.05   206.3 3817.65
   210.1 3818.62   222.6 3821.65   227.2 3822.37   251.1 3822.62   267.4 3823.47
   283.5 3822.89   319.9 3821.97     336 3822.43     340 3822.73   344.1  3823.7
   352.1 3826.25   360.2 3827.73   368.3 3828.06   376.3 3828.84   388.7  3828.8
#Mann= 5 ,-1,0
       0     .12       0    61.4      .1       0151.9205    .045       0
   210.1     .12       0   283.5      .1       0
Bank Sta=151.9205,210.1
XS Rating Curve= 0 ,0
Exp/Cntr(USF)=0,0
Exp/Cntr=0.3,0.1

Type RM Length L Ch R = 1 ,30110   ,266.4,268.8,272.9
XS GIS Cut Line= 2
2266869.04418469536667.6946444062267210.24354606536715.582274071
#Sta/Elev= 30
       0 3843.15    11.2 3841.46    27.4 3837.75    39.5 3833.34    59.7 3821.31
    67.8 3817.28    71.8 3815.84    75.9 3815.18    96.1 3815.06   103.3 3815.24
   106.8 3815.74     110 3816.11   128.4 3818.15   140.5 3817.41   145.8 3817.62
   149.3    3818   160.7 3820.44     193 3817.78   213.1 3819.83   221.3 3820.62
   241.6 3820.81   253.6 3820.39   265.7 3819.05   281.9 3820.49     294 3820.52
   298.1 3821.21   306.1 3823.86   318.2 3824.92   326.3 3826.25   344.5 3826.01
#Mann= 6 ,-1,0
       0     .12       0    27.4      .1       0    71.8    .045       0
   106.8      .1       0     110     .12       0   213.1      .1       0
Bank Sta=71.8,106.8
XS Rating Curve= 0 ,0
Exp/Cntr(USF)=0,0
Exp/Cntr=0.3,0.1

Type RM Length L Ch R = 1 ,29842   ,340.2,358.5,392.9
XS GIS Cut Line= 2
2266817.16591922536917.1093822472267130.43082995 536998.91741626
#Sta/Elev= 30
       0 3830.32    11.4 3829.22    15.5 3828.48    23.8 3826.35    36.2 3823.66
    65.1 3820.18    77.5  3819.9   100.9 3814.46   106.5 3813.88   131.3 3813.91
   136.9 3814.34   143.7 3815.15   156.1 3815.67   160.2 3816.19   164.3 3817.23
     185  3817.7   202.5 3816.93     214 3817.52   230.5 3817.28   251.2 3818.54
   259.4 3818.17   271.8 3818.34     276 3818.67   277.9 3819.11   280.1 3819.69
   284.4 3821.46   288.4 3822.39   300.8 3824.16   313.9 3825.46   323.8 3825.95
#Mann= 4 ,-1,0
       0     .12       0   100.9    .045       0   136.9     .12       0
     270      .1       0
Bank Sta=100.9,136.9
XS Rating Curve= 0 ,0
Exp/Cntr(USF)=0,0
Exp/Cntr=0.3,0.1

Type RM Length L Ch R = 1 ,29483   ,174.5,174.8,174.5
XS GIS Cut Line= 2
2266711.41407037537014.8799594812266809.18464761537380.023135682
#Sta/Elev= 30
       0 3823.94     6.5 3822.93    23.1 3821.85    31.4  3820.9    35.5  3820.9
      45 3822.18    60.4 3822.33    85.2 3820.11   122.5 3818.59     143 3818.15
   155.6 3817.37   192.9 3816.75   213.6 3814.82     226 3814.65     251 3812.79
   259.1 3812.12   271.5 3812.05   279.8 3812.33   281.3 3812.83     284 3813.78
   292.2 3819.41   296.2 3821.59   300.5 3822.72   308.8 3824.23   325.4 3825.43
   346.1 3826.13   350.2 3827.06   362.6 3833.91   366.8 3834.83     378 3835.02
#Mann= 4 ,-1,0
       0     .12       0     220      .1       0     251    .045       0
   281.3      .1       0
Bank Sta=251,281.3
XS Rating Curve= 0 ,0
Exp/Cntr(USF)=0,0
Exp/Cntr=0.3,0.1

Type RM Length L Ch R = 1 ,29308   ,222.8,226.7,231.6
XS GIS Cut Line= 2
2266545.80268445537070.7488607582266643.57326168537431.901401153
#Sta/Elev= 30
       0 3829.35    27.4 3823.07    46.3 3822.01    68.3 3819.19    75.7 3817.78
    81.3 3817.25   108.3 3816.44   143.4 3816.64   155.8 3817.26   176.6    3817
   222.1  3815.3   234.6 3814.18   245.2 3811.98     247 3811.61     255 3811.35
   280.2 3811.49   282.33812.004   284.4 3812.53   288.5 3815.47   292.6 3818.99
   296.7  3821.3   300.9 3822.74     305 3823.51   321.6 3824.61   346.5 3823.69
   350.6 3825.08   354.8 3827.73   358.9 3829.41   371.3 3831.53   374.2 3831.65
#Mann= 4 ,-1,0
       0      .1       0     150     .12       0   245.2    .045       0
   282.3      .1       0
Bank Sta=245.2,282.3
XS Rating Curve= 0 ,0
Exp/Cntr(USF)=0,0
Exp/Cntr=0.3,0.1

Type RM Length L Ch R = 1 ,29082   ,189.1,173.8,161.1
XS GIS Cut Line= 2
 2266368.2193911537156.5475305762266406.13043126537501.737527748
#Sta/Elev= 30
       0 3836.37     4.7 3836.02    36.8 3830.98    52.9 3827.76    64.1  3826.8
    73.1 3825.09    83.9 3824.29   117.3 3821.06   125.4 3820.74   133.4 3819.44
   141.5 3816.77   145.4 3815.95   157.6  3814.5   173.7 3813.84   181.7 3811.45
   185.7 3811.41   189.8 3810.89   218.1 3810.56   226.8 3810.77   246.1 3812.97
   254.2 3814.34   270.2 3814.16   282.3 3815.37     287 3816.47   294.2 3820.11
   298.4 3821.88   302.4 3822.94   306.5 3823.61   326.9 3824.15   347.3 3823.19
#Mann= 3 ,-1,0
       0      .1       0   189.8    .045       0   226.8      .1       0
Bank Sta=189.8,226.8
XS Rating Curve= 0 ,0
Exp/Cntr(USF)=0,0
Exp/Cntr=0.3,0.1

Type RM Length L Ch R = 1 ,28908   ,210.6,196.9,185.6
XS GIS Cut Line= 2
2266140.75315019 537276.266604742266328.31303305537549.625157414
#Sta/Elev= 30
       0  3855.6       6 3853.89    15.7 3851.97    39.9 3846.21    69.3 3837.57
    76.7 3834.88    88.4 3829.09   109.6 3815.97   117.5 3810.56   119.2 3810.01
   122.4 3809.27   138.3 3809.07   151.5 3809.42   156.3 3809.91   161.2 3810.95
     166 3811.19   175.7  3812.5   195.1 3812.83   213.1 3812.34   241.9 3815.51
   253.4 3815.78   273.6 3815.14   282.5 3816.51   287.3 3818.72   292.2 3821.61
   296.6 3823.23   299.4 3823.71   305.2 3824.28   322.5 3824.48   331.5 3823.83
#Mann= 3 ,-1,0
       0      .1       0   119.2    .045       0   156.3      .1       0
Bank Sta=119.2,156.3
XS Rating Curve= 0 ,0
Exp/Cntr(USF)=0,0
Exp/Cntr=0.3,0.1

Type RM Length L Ch R = 1 ,28711   ,235.3,223.6,211.5
XS GIS Cut Line= 2
2265991.10430749537481.7843487212266250.49563484537635.423827232
#Sta/Elev= 30
       0 3853.15     5.9 3851.24    10.5 3849.02    14.5 3847.53    33.8 3842.03
    38.4 3839.95    45.9 3835.64    47.7 3835.02    61.7 3831.89    67.5 3829.97
    76.3 3825.71    87.9 3818.23    94.2 3814.65   103.5 3810.26   108.2 3808.94
     120 3808.45   136.1 3808.31   149.2  3808.8   154.7 3809.26   173.3 3815.13
   179.3 3815.11   201.8 3812.66   228.1 3814.92     250 3815.34   252.3 3815.56
   257.3 3817.09     266 3821.57   271.9 3823.03   289.2    3824   301.5 3823.33
#Mann= 3 ,-1,0
       0      .1       0   108.2    .045       0   149.2      .1       0
Bank Sta=108.2,149.2
XS Rating Curve= 0 ,0
Exp/Cntr(USF)=0,0
Exp/Cntr=0.3,0.1

Type RM Length L Ch R = 1 ,28487   ,348.6,347.1,343.2
XS GIS Cut Line= 2
2265919.27286299537743.1709939792266160.70632922537779.086716229
#Sta/Elev= 30
       0 3847.81       5 3845.86      13 3842.06    25.2 3835.71    30.7 3832.55
    37.8 3829.02    45.4 3824.94    51.8  3822.5    85.8 3812.03    89.9 3811.45
    93.9 3811.32   106.1 3809.68   114.1  3807.7   118.2 3807.18   126.3 3807.28
   146.5 3806.94   153.9 3807.14   158.6 3807.57   162.7 3808.97   174.8 3813.69
   182.9  3816.4   189.1 3818.12     195 3819.27   203.9 3819.54   207.2 3820.03
   215.2 3822.03   219.3 3822.51   227.4 3822.23   235.5 3822.67   244.1 3822.07
#Mann= 3 ,-1,0
       0      .1       0   114.1    .045       0   158.6      .1       0
Bank Sta=114.1,158.6
XS Rating Curve= 0 ,0
Exp/Cntr(USF)=0,0
Exp/Cntr=0.3,0.1

Type RM Length L Ch R = 1 ,28140   ,169.7,169.3,169
XS GIS Cut Line= 2
 2265855.4226901538092.3516269582266106.83274584538112.304805985
#Sta/Elev= 30
       0 3828.02     8.8  3826.1      13 3824.73    36.9 3818.85    44.9 3817.14
    52.9 3815.07      77 3810.12      85 3808.82      89 3808.52    97.1 3808.34
   101.1 3808.78   105.1 3808.11   109.3 3807.07   113.1 3806.56   117.1 3806.49
   153.2 3806.42   161.3 3806.56   162.1 3806.89   165.5 3808.15   177.3 3811.16
   189.3 3813.85   193.4 3814.43   209.4 3814.94   225.5 3814.96   229.5 3815.26
   233.5 3816.06   237.5 3817.46   241.5 3818.15   249.5 3818.13   252.2 3818.33
#Mann= 4 ,-1,0
       0      .1       0   109.3    .045       0   162.1      .1       0
     240     .08       0
Bank Sta=109.3,162.1
XS Rating Curve= 0 ,0
Exp/Cntr(USF)=0,0
Exp/Cntr=0.3,0.1

Type RM Length L Ch R = 1 ,27971   ,199.4,181.5,162.1
XS GIS Cut Line= 3
2265835.46951107 538261.953648692266100.84679214538279.911509815
 2266148.7344218538259.958330787
#Sta/Elev= 30
       0 3840.27    16.7 3832.17    26.2 3828.39    32.8 3826.04    36.8 3824.31
    40.8 3823.31    60.8 3820.13    64.9 3819.51    68.9 3819.22    80.9 3817.26
    84.9 3816.17     109 3807.04     122 3805.84     149 3805.65   157.1 3805.84
   159.93807.099   165.1 3808.75   173.1 3808.98   197.2 3811.13   253.3 3812.25
   261.3 3812.87   265.3 3813.09   278.3 3812.66   282.6 3812.88   286.9 3814.32
   291.3 3816.12   295.6 3817.08   304.3 3817.25   312.9 3818.25   317.9 3818.12
#Mann= 5 ,-1,0
       0      .1       0    60.8     .12       0     109    .045       0
   159.9     .12       0   261.3      .1       0
Bank Sta=109,159.9
XS Rating Curve= 0 ,0
Exp/Cntr(USF)=0,0
Exp/Cntr=0.3,0.1

Type RM Length L Ch R = 1 ,27789   ,210.1,209.3,208.8
XS GIS Cut Line= 2
2265901.31500186538511.3683865322266166.69228293  538341.7663648
#Sta/Elev= 30
       0 3821.86     3.7 3821.09     8.1 3820.59    18.9 3820.17    36.6 3818.86
    47.1 3817.38    73.2 3815.32      79 3814.63    84.1 3813.64     105 3805.47
   107.9 3804.79   112.6 3804.73   128.2 3804.75   136.3  3805.5   141.1 3805.77
   150.6 3807.62   165.8 3809.57     179 3810.35     198 3808.91   207.5 3810.04
   234.3  3810.9   245.5 3810.84   264.5 3809.79   269.2  3809.9     274 3810.35
   283.5 3812.18   297.7 3816.14   301.2 3816.85   307.2 3817.05   314.9 3817.98
#Mann= 3 ,-1,0
       0     .12       0     105    .045       0   136.3     .12       0
Bank Sta=105,136.3
XS Rating Curve= 0 ,0
Exp/Cntr(USF)=0,0
Exp/Cntr=0.3,0.1

Type RM Length L Ch R = 1 ,27580   ,180,182.3,184.6
XS GIS Cut Line= 2
 2265999.0855791538698.9282693892266250.49563484538533.316883462
#Sta/Elev= 30
       0 3816.57    10.9 3816.47      30 3815.88    54.1 3814.53    59.8 3814.98
    68.6 3816.14    82.7 3815.28    91.6 3813.74    94.5 3812.35    97.1 3810.54
   100.2  3809.1     106 3806.73   112.3 3804.86   117.6 3804.22   143.5 3804.08
   154.33804.741   189.7 3807.48   207.3 3807.82   231.2 3809.94   236.3 3810.05
   256.2 3808.82   259.1 3808.97     260  3809.1   264.4 3811.17   270.6 3814.82
   274.3 3816.17   279.1  3816.9   286.8 3817.19   293.5 3817.93   301.1 3817.76
#Mann= 6 ,-1,0
       0      .1       0      10     .12       0   112.3    .045       0
   154.3      .1       0     190     .12       0     230      .1       0
Bank Sta=112.3,154.3
XS Rating Curve= 0 ,0
Exp/Cntr(USF)=0,0
Exp/Cntr=0.3,0.1

Type RM Length L Ch R = 1 ,27398   ,232.5,243.6,255.5
XS GIS Cut Line= 3
2266023.02939393538808.6707540392266158.71101132538806.675436137
2266340.28494047   538706.909541
#Sta/Elev= 30
       0 3816.71    13.1 3813.51    25.1 3813.41    37.1 3812.29    51.9 3813.25
    57.2 3813.06    70.7 3810.68    81.2 3809.32    93.2 3809.39   101.2 3810.33
   141.9 3811.65   149.7 3810.03     172  3803.6   178.4 3803.22   201.3 3803.17
   205.8 3803.21   208.6 3803.67     215 3806.03   219.5 3806.75   230.2 3806.51
   255.7 3807.75   273.4 3806.28   278.9 3806.33   285.2 3807.79   296.9 3812.91
   308.7 3815.43   315.4 3815.68   324.5 3817.07   329.1 3817.18   342.9 3816.45
#Mann= 5 ,-1,0
       0      .1       0      70     .12       0   165.7      .1       0
     172    .045       0   208.6     .12       0
#XS Ineff= 2 , 0
          140.54 3812.56
Permanent Ineff=
       F       F
Bank Sta=172,208.6
XS Rating Curve= 0 ,0
Exp/Cntr(USF)=0,0
Exp/Cntr=0.3,0.1

Type RM Length L Ch R = 1 ,27154   ,293,309.8,325.5
XS GIS Cut Line= 3
2266027.02002974 539006.207226412266160.70632922539026.160405437
2266374.20534481539004.211908507
#Sta/Elev= 30
       0 3812.71    13.3  3811.8    33.5 3809.92    45.7 3809.48    53.7 3810.05
      78 3808.23    86.1 3808.03   102.3 3808.37   114.4 3809.14   126.5 3809.48
   154.7 3809.63   170.8 3808.64     183 3808.53   197.6 3807.96   204.9 3807.22
   218.6 3803.39     223 3802.73   231.1 3802.14   255.3 3802.32   262.1 3802.76
   295.5 3805.26   299.7 3806.13   303.5 3807.31   315.6 3813.53   319.6 3814.28
   323.6 3814.38   331.7 3816.06   339.7 3816.41   347.8 3815.12   349.8 3815.22
#Mann= 5 ,-1,0
       0     .12       0      70      .1       0  165.17     .12       0
     223    .045       0   262.1     .12       0
#XS Ineff= 2 , 0
          156.61 3811.38
Permanent Ineff=
       F       F
Bank Sta=223,262.1
XS Rating Curve= 0 ,0
Exp/Cntr(USF)=0,0
Exp/Cntr=0.3,0.1

Type RM Length L Ch R = 1 ,26844   ,394.1,368.3,322.7
XS GIS Cut Line= 2
2265961.17453895539205.7390166832266304.36921822539365.364448902
#Sta/Elev= 30
       0 3814.72     7.7 3814.78    16.5 3814.42    34.2 3812.78    60.7  3812.4
    69.5 3811.93    82.7 3811.93    93.5  3811.1   100.4 3810.88   113.6 3809.05
   126.8  3809.2   148.9 3808.44   162.1 3808.68   179.8 3807.86   197.6 3805.02
   206.2 3802.37   210.6 3801.61   218.6 3801.15   250.4 3801.22   257.8 3801.53
   276.8  3805.1   290.1 3804.68   294.5 3804.87   302.2    3806     315 3808.77
     318 3809.15     343 3809.25   351.1 3809.67   360.1 3810.58   378.5 3810.49
#Mann= 6 ,-1,0
       0     .12       0     190      .1       0   210.6    .045       0
   257.8      .1       0     260     .12       0     370      .1       0
#XS Ineff= 2 , 0
          161.17 3810.42
Permanent Ineff=
       F       F
Bank Sta=210.6,257.8
XS Rating Curve= 0 ,0
Exp/Cntr(USF)=0,0
Exp/Cntr=0.3,0.1

Type RM Length L Ch R = 1 ,26476   ,290.8,263.8,218
XS GIS Cut Line= 3
2266048.96852667539722.5263534912266268.45349597539483.088205163
2266314.86522344539394.672250901
#Sta/Elev= 30
       0 3816.34    12.7 3816.11    40.3 3814.89    61.5 3815.27    77.8 3813.75
    83.2 3812.91    88.2 3811.45   104.9 3801.51     108 3800.37   110.8 3799.76
   121.2 3799.69   136.3  3799.7   140.9  3800.3   147.6 3802.55   153.8 3803.32
   170.5 3803.62   178.8 3802.99   201.4 3804.02   213.5 3803.99   223.8 3804.62
   252.4 3805.08   312.6 3807.91   324.4 3807.62   341.4  3807.7   349.7 3808.05
   372.1 3807.64   385.7 3808.27   400.1 3807.47   420.8 3809.71   424.7 3809.84
#Mann= 3 ,-1,0
       0     .12       0     108    .045       0   140.9     .12       0
#XS Ineff= 2 , 0
                          313.25         3813.23
Permanent Ineff=
       F       F
Bank Sta=108,140.9
XS Rating Curve= 0 ,0
Exp/Cntr(USF)=0,0
Exp/Cntr=0.3,0.1

Type RM Length L Ch R = 1 ,26212   ,109.2,119.1,126.2
BEGIN DESCRIPTION:
Structure XS 4
END DESCRIPTION:
XS GIS Cut Line= 2
2266458.00869673539730.5076251032266276.43476758539491.069476774
#Sta/Elev= 30
       0 3826.13    21.7 3824.64    26.8 3824.12    45.1 3820.26      77 3814.74
    90.8 3813.46   102.1 3812.72   117.1 3809.06   132.2 3803.97   142.2 3801.36
   148.7 3799.98   161.33798.362   168.5 3798.04   179.3 3797.99   188.4 3798.13
   190.7 3798.32   197.5 3799.48   202.5 3801.04   207.5 3802.14   216.4 3801.46
   222.1  3801.6   227.6 3801.95   232.6 3803.19   239.2 3805.11   242.6 3805.81
   259.2 3806.18   267.7 3806.71   273.5 3806.42   287.8 3806.56   300.5 3807.25
#Mann= 4 ,-1,0
       0      .1       0      70     .12       0   161.3    .045       0
   190.7     .12       0
Bank Sta=161.3,190.7
XS Rating Curve= 0 ,0
Exp/Cntr(USF)=0,0
Exp/Cntr=0.5,0.3
