HEC-RAS study SHVRSFK.prj: SHVRSFK

--- SHVRSFK.g01 (geometry) --- (continued)

Type RM Length L Ch R = 1 ,26093   ,67.3,66.8,64.1
BEGIN DESCRIPTION:
Structure XS 3
END DESCRIPTION:
XS GIS Cut Line= 2
  2266513.877598539720.5310355892266390.16788803539379.331674221
#Sta/Elev= 30
       0 3819.25    16.3 3821.68    29.1 3822.98    40.2 3822.98    58.9 3820.35
    63.1 3818.82    71.6 3814.19    80.2 3811.18    88.7 3809.91   105.7 3806.08
   118.4 3802.21   145.8 3801.88   165.2 3802.29     181 3801.06   190.8 3801.28
     195 3800.71   206.9 3797.33   228.8 3796.94   241.8 3797.14   254.6 3800.66
   258.9 3801.13   267.4 3801.07   278.7 3803.35   284.4 3803.84   292.9 3806.19
   305.7 3806.76   326.9 3809.73   335.4 3809.41   348.2 3810.86   362.9 3810.39
#Mann= 5 ,-1,0
       0     .12       0      50      .1       0      90     .12       0
   206.9    .045       0   241.8     .12       0
#XS Ineff= 2 , 0
             173    3812     277            3813
Permanent Ineff=
       F       F
Bank Sta=206.9,241.8
XS Rating Curve= 0 ,0
Exp/Cntr(USF)=0,0
Exp/Cntr=0.5,0.3

Type RM Length L Ch R = 1 ,26026   ,166.4,172.5,180
BEGIN DESCRIPTION:
Structure XS 2
END DESCRIPTION:
XS GIS Cut Line= 2
 2266581.7184067539710.5544460752266448.03210721539357.383177291
#Sta/Elev= 30
       0 3808.28     5.7 3808.53    14.7 3809.72    31.4  3812.5      40 3812.99
    69.9 3813.27      87 3812.07   116.7 3804.34   125.5 3801.69   129.8 3801.05
   159.7 3800.47   168.3 3800.78   179.1 3800.11   185.4 3800.35   193.9 3801.33
   202.5  3801.4   223.9 3800.32   240.6 3797.19   249.5 3796.83   264.2 3797.24
   270.9 3798.21   279.5 3801.22   300.9 3801.73   305.1 3802.77   315.6 3807.83
   321.8 3809.28   339.4 3810.92   356.5 3811.08   369.3 3812.77   377.6 3812.99
#Mann= 5 ,-1,0
       0     .12       0      40      .1       0   240.6    .045       0
   264.2      .1       0     280     .12       0
#XS Ineff= 2 , 0
             218    3812     292            3813
Permanent Ineff=
       F       F
Bank Sta=240.6,264.2
XS Rating Curve= 0 ,0
Exp/Cntr(USF)=0,0
Exp/Cntr=0.5,0.3

Type RM Length L Ch R = 1 ,25854   ,211.1,238.7,260.6
BEGIN DESCRIPTION:
Structure XS 1
END DESCRIPTION:
XS GIS Cut Line= 3
2266667.51707651539680.6246775342266667.51707651539509.027337899
2266633.59667217539299.518958112
#Sta/Elev= 30
       0 3805.91     7.4 3806.24    19.4  3805.9    39.4 3806.81    67.4  3805.8
    75.4 3804.84    87.4 3804.45   107.4 3800.92   119.4 3799.74   131.4 3797.74
   135.4 3797.61   151.4 3799.38   179.5 3800.59   195.8 3799.19     216 3800.03
   236.3 3799.88   247.6 3796.79   254.4 3796.56   280.9 3796.22   297.1 3796.51
   301.1 3796.85   305.2 3798.11   317.3 3806.82   325.4 3811.23   329.5 3812.47
   337.6 3812.76   353.8  3814.7   365.9  3817.6   378.1 3819.68   383.8 3821.14
#Mann= 6 ,-1,0
       0      .1       0      10     .12       0     110      .1       0
   254.4    .045       0   297.1      .1       0   301.6     .12       0
Bank Sta=254.4,297.1
XS Rating Curve= 0 ,0
Exp/Cntr(USF)=0,0
Exp/Cntr=0.3,0.1

Type RM Length L Ch R = 1 ,25615   ,73.5,111.2,131.1
XS GIS Cut Line= 2
2266715.40470618539686.6106312422266926.90840387539397.289535346
#Sta/Elev= 30
       0  3805.4     8.1 3805.85    38.8 3805.32      56 3805.57    66.2  3804.7
    81.7 3804.37   101.8 3801.55   118.9 3801.68   130.6  3799.5     139 3799.61
   155.4 3801.15   173.3 3798.87   196.2 3797.62   218.2 3797.55   224.8 3796.19
   232.33795.224   247.7 3794.58   274.13795.177   282.1 3796.02   290.7 3797.45
   294.1 3798.64   299.5  3802.5     304 3804.62   318.9 3806.93   326.6 3811.05
   328.8 3811.87   333.6 3812.46   340.2 3812.48   345.1 3813.38   358.4 3819.17
#Mann= 4 ,-1,0
       0     .12       0   232.3    .045       0   274.1      .1       0
     280     .12       0
Bank Sta=232.3,274.1
XS Rating Curve= 0 ,0
Exp/Cntr(USF)=0,0
Exp/Cntr=0.3,0.1

Type RM Length L Ch R = 1 ,25504   ,156.1,167.5,177.8
XS GIS Cut Line= 3
2266724.27095573539683.6269162472266825.18179913539576.320848144
2267054.33350602539585.869536701
#Sta/Elev= 30
       0 3805.71     7.3 3805.13    14.3 3805.39    35.6 3804.58    52.8 3805.49
    66.7 3804.42    75.8 3804.38    93.3 3801.48     112 3801.84   117.7 3801.53
   124.2 3800.34   129.7 3799.89   158.3 3800.85   166.4 3799.77   178.3 3797.35
   198.3 3794.75   206.3 3794.11   220.5  3794.2   228.9 3794.62   250.4 3795.67
   266.3 3804.44   270.1 3806.32   274.4 3807.85   286.4 3809.86   298.4 3810.97
   310.4 3816.05   314.4 3817.05   354.5 3824.25   366.2 3826.84   376.7 3828.36
#Mann= 4 ,-1,0
       0     .12       0   198.3    .045       0   228.9     .12       0
   307.3      .1       0
Bank Sta=198.3,228.9
XS Rating Curve= 0 ,0
Exp/Cntr(USF)=0,0
Exp/Cntr=0.3,0.1

Type RM Length L Ch R = 1 ,25336   ,209.6,217.6,228.4
XS GIS Cut Line= 2
 2266729.3719315539690.6012670482266958.83349031539792.362480087
#Sta/Elev= 30
       0 3805.31     3.1 3805.15    13.2 3805.27    26.1 3804.22    42.4 3803.27
    55.6 3802.82      60 3801.85    81.8  3796.4    90.6 3793.51      95 3793.09
   125.6 3792.94   131.4 3792.99   134.3 3793.12   136.53793.399   138.7 3793.82
   143.1 3795.48   144.5 3795.77   156.2 3796.91     165    3797   179.9 3799.57
   195.6 3802.87   201.1  3804.4   204.3 3805.47   208.7 3806.24   217.5 3807.35
   233.3 3810.57   240.5 3812.25   243.6 3812.84   248.1 3813.34     251 3813.91
#Mann= 4 ,-1,0
       0     .12       0    90.6    .045       0   136.5     .12       0
     220      .1       0
Bank Sta=90.6,136.5
XS Rating Curve= 0 ,0
Exp/Cntr(USF)=0,0
Exp/Cntr=0.3,0.1

Type RM Length L Ch R = 1 ,25119   ,81.9,94.2,118.6
BEGIN DESCRIPTION:
Structure XS 4
END DESCRIPTION:
XS GIS Cut Line= 3
2266625.61540056539792.362480087 2266659.5358049539868.184560391
2266918.92713226540073.702304373
#Sta/Elev= 30
       0 3804.55    22.8 3804.17    44.7  3803.1    57.1  3803.3    75.2 3802.72
    83.9 3802.86    89.9 3802.25    97.5  3802.1   110.4 3799.79   124.1 3798.32
     140 3796.04   155.5 3795.05   165.33793.081   169.6  3792.4   175.3 3792.03
   196.2 3791.94   213.5 3792.39   216.6 3792.62   219.53793.318     238 3800.89
   255.1 3804.16   263.6  3805.1   280.7 3810.04   303.5 3815.96   323.4 3821.75
   357.6 3829.27     381  3835.8   391.7  3838.3   400.3 3839.91     414 3843.27
#Mann= 6 ,-1,0
       0     .12       0  103.06      .1       0  113.06     .12       0
   165.3    .045       0   219.5     .12       0  373.06      .1       0
Bank Sta=165.3,219.5
XS Rating Curve= 0 ,0
Exp/Cntr(USF)=0,0
Exp/Cntr=0.5,0.3

Type RM Length L Ch R = 1 ,25025   ,85.5,87.6,85
BEGIN DESCRIPTION:
Structure XS 3
END DESCRIPTION:
XS GIS Cut Line= 3
2266610.81871106539785.0874039972266702.60333458540080.394453602
2266698.61269878540255.982429042
#Sta/Elev= 30
       0 3805.89      21 3804.69    29.4 3804.73    46.2 3803.59   100.6    3802
   117.4 3800.64   141.8 3799.97   166.3  3795.8   176.9 3795.74   192.9 3794.77
   205.7 3793.35   218.5 3791.17     244 3790.53   255.6 3790.61     260 3791.07
   268.2 3796.23   272.8 3798.29   279.2 3800.47   289.1 3802.95   305.9 3804.22
     310 3804.18     318 3803.21     338 3805.49   373.1  3803.5     390 3804.29
   402.1 3802.98   410.1 3803.85   438.1 3803.11   446.1 3802.42   484.9 3802.21
#Mann= 6 ,-1,0
       0     .12       0     100      .1       0     200     .12       0
   218.5    .045       0     260      .1       0  309.24     .12       0
#XS Ineff= 2 , 0
             182  3807.5     298          3805.5
Permanent Ineff=
       F       F
Bank Sta=218.5,260
XS Rating Curve= 0 ,0
Exp/Cntr(USF)=0,0
Exp/Cntr=0.5,0.3

Type RM Length L Ch R = 1 ,24937   ,230,199.2,166.7
BEGIN DESCRIPTION:
Structure XS 2
END DESCRIPTION:
XS GIS Cut Line= 3
2266541.81204864539836.2594739472266633.59667217540131.566523552
2266625.61540056540231.332418689
#Sta/Elev= 30
       0 3809.26     9.3 3808.93    17.7 3807.15    38.7 3806.42    59.6 3803.87
    76.4 3802.63    97.3 3801.88   114.1 3800.12   151.8 3799.63   160.1 3799.15
   184.8 3795.63   194.4 3795.57   206.2 3793.33   214.6 3791.08   218.8 3790.66
   239.7 3790.51   253.1 3790.92   256.5 3791.46   261.5 3793.34   264.7 3794.18
   273.2 3794.96   290.2 3799.52   306.7 3801.16   319.5 3801.31     359 3800.51
   371.1 3800.96   378.9 3800.68   395.1 3800.88   403.2 3800.52   409.3 3800.65
#Mann= 4 ,-1,0
       0      .1       0     150     .12       0   214.6    .045       0
   253.1     .12       0
#XS Ineff= 2 , 0
           200.7  3807.5   279.3          3805.5
Permanent Ineff=
       F       F
Bank Sta=214.6,253.1
XS Rating Curve= 0 ,0
Exp/Cntr(USF)=0,0
Exp/Cntr=0.5,0.3

Type RM Length L Ch R = 1 ,24738   ,166.7,167.7,169.5
BEGIN DESCRIPTION:
Structure XS 1
END DESCRIPTION:
XS GIS Cut Line= 2
2266318.33644354540201.4026501482266593.69031411540241.309008202
#Sta/Elev= 30
       0 3854.61     9.9 3852.73      14  3851.7      18 3850.11    22.1 3848.17
    42.3 3836.32    46.3 3834.73    50.4 3832.68    58.4 3826.36    62.5 3824.23
    78.7 3819.32    94.8 3813.31    98.9 3812.52     111 3808.76   117.9 3806.92
   123.1 3805.79   134.8 3803.86   151.4 3799.72   156.8 3798.03   167.3 3793.75
   178.43790.401   183.7 3789.47   191.8 3789.59   203.9 3789.39   213.2 3790.11
   224.2 3791.43   236.3 3795.17   248.5 3797.89   260.5 3799.29   278.2 3799.41
#Mann= 4 ,-1,0
       0      .1       0      70     .12       0   178.4    .045       0
   213.2     .12       0
Bank Sta=178.4,213.2
XS Rating Curve= 0 ,0
Exp/Cntr(USF)=0,0
Exp/Cntr=0.3,0.1

Type RM Length L Ch R = 1 ,24570   ,359.3,363,367.1
XS GIS Cut Line= 2
2266310.35517192540365.0187181722266607.65753943 540414.90166574
#Sta/Elev= 30
       0 3839.73     5.9 3838.47      10 3837.01    18.1 3832.66    22.1 3831.09
    42.4 3824.53    62.7  3816.5    75.1 3811.84      87 3809.26   103.2 3807.12
   121.8 3806.43   127.6 3805.75   131.6 3804.95   138.5  3802.7   151.9 3797.88
   164.1 3791.49   168.1 3789.69   172.2 3789.06   188.4 3789.02   212.8 3789.06
   218.5 3789.59     229 3790.87   242.7 3792.19   269.2 3795.48   273.6 3796.64
   277.6 3798.74   281.7 3800.17     290 3801.21   296.9 3802.46   301.5 3802.47
#Mann= 4 ,-1,0
       0     .12       0      20      .1       0   168.1    .045       0
   218.5      .1       0
Bank Sta=168.1,218.5
XS Rating Curve= 0 ,0
Exp/Cntr(USF)=0,0
Exp/Cntr=0.3,0.1

Type RM Length L Ch R = 1 ,24207   ,261.4,257.8,252.5
XS GIS Cut Line= 2
2266240.51904533540700.2321258312266535.82609493540784.035477746
#Sta/Elev= 30
       0 3800.04       8 3799.45    20.4 3797.56    36.1 3797.08    56.2 3796.81
   117.1 3796.77   120.3 3796.48   139.8 3791.64   145.2 3789.67   148.53787.903
   149.5 3787.42   153.5 3787.16   190.9 3787.19   195.1 3787.32   197.43787.765
   203.4 3789.46   211.7 3790.65   233.7 3792.03   253.3 3794.48   257.4 3795.55
   261.6 3797.71   265.8 3798.95   274.1 3799.45   278.2 3800.13   282.4 3800.25
   286.5 3799.83   290.7 3798.72   294.9 3798.18     299 3798.82     307 3801.34
#Mann= 3 ,-1,0
       0      .1       0   148.5    .045       0   197.4      .1       0
Bank Sta=148.5,197.4
XS Rating Curve= 0 ,0
Exp/Cntr(USF)=0,0
Exp/Cntr=0.3,0.1

Type RM Length L Ch R = 1 ,23949   ,136.6,133.8,130.2
XS GIS Cut Line= 3
2266102.84211004540917.7217772292266236.52840952540981.571950117
  2266513.877598541021.478308172
#Sta/Elev= 30
       0 3799.47       8 3798.48    17.3 3798.07    36.9 3796.11    63.4 3794.54
    76.8  3794.2    99.6 3794.29   112.3 3795.37   125.6 3795.93   143.3 3796.15
     168 3795.74   192.2 3793.75   200.5 3793.45   236.7 3787.44   244.93787.004
   264.1 3786.62   285.2 3786.66   289.2 3787.04   297.3 3789.09   301.4 3789.08
   309.4 3789.95   313.4 3790.74   321.6 3793.34   345.8 3796.37   353.9 3796.89
   370.1 3799.41   378.1 3798.75   382.2 3797.35   386.2 3796.86   428.4 3806.98
#Mann= 4 ,-1,0
       0      .1       0  208.15     .12       0   244.9    .045       0
   289.2     .12       0
Bank Sta=244.9,289.2
XS Rating Curve= 0 ,0
Exp/Cntr(USF)=0,0
Exp/Cntr=0.3,0.1

Type RM Length L Ch R = 1 ,23815   ,156.8,155.2,153.9
XS GIS Cut Line= 3
2266059.75271615541116.2560698542266464.92824368541137.522188702
2266541.03856376541101.705567485
#Sta/Elev= 30
       0 3798.39    44.5 3792.23    80.5 3792.11    88.5 3791.14   140.6 3794.24
   176.7 3791.68   216.7 3792.46   228.7 3790.87   237.2 3790.57   260.1 3786.43
   268.8 3785.85   300.8 3785.94   303.8 3786.45   308.8 3787.82   320.9 3789.66
   364.9 3793.57   372.9 3795.24   376.9 3795.47     385 3794.24     389 3794.85
   396.8 3797.26     405 3798.68   409.3  3798.6   418.2  3796.4   423.5 3796.19
   435.5  3796.4   459.5 3798.18   471.6 3799.84   484.5  3802.9   489.8 3804.67
#Mann= 4 ,-1,0
       0      .1       0   260.1    .045       0   303.8      .1       0
  435.73     .12       0
#XS Ineff= 2 , 0
          201.46 3795.15
Permanent Ineff=
       F       F
Bank Sta=260.1,303.8
XS Rating Curve= 0 ,0
Exp/Cntr(USF)=0,0
Exp/Cntr=0.3,0.1

Type RM Length L Ch R = 1 ,23660   ,279.2,258.3,234.2
XS GIS Cut Line= 4
2266094.32588175541378.7830245222266250.25814467541284.142590957
2266475.96655785541288.850907138 2266581.7184067541219.014780542
#Sta/Elev= 30
       0 3833.96    11.5 3828.62    25.8  3822.8    58.3 3805.89    72.3 3799.15
      77 3797.12    95.7 3792.43     111 3789.72   121.9 3788.84   153.9 3788.17
     180 3788.28   208.3 3786.64   220.3 3786.84228.77273786.028   240.2 3785.47
   284.3 3785.41292.05893786.118   304.3 3789.48   324.4 3792.34   367.2 3792.72
     393 3793.68   432.4 3793.66   437.2 3794.01   446.8 3796.39   456.3 3797.41
   474.5 3796.02   480.3 3794.71   494.7 3793.97   509.1 3795.28   534.9 3796.01
#Mann= 5 ,-1,0
       0     .12       0     120      .1       0228.7727    .045       0
292.0589      .1       0  428.16     .12       0
#XS Ineff= 2 , 0
          104.73 3794.48   323.2         3801.61
Permanent Ineff=
       F       F
Bank Sta=228.7727,292.0589
XS Rating Curve= 0 ,0
Exp/Cntr(USF)=0,0
Exp/Cntr=0.3,0.1

Type RM Length L Ch R = 1 ,23402   ,245.4,234.2,222.9
XS GIS Cut Line= 2
 2266220.5658663541638.0315401162266631.60135426 541348.71044422
#Sta/Elev= 30
       0 3850.18    15.4 3842.13    26.2 3839.49    43.5 3836.87      52 3834.74
   103.7 3814.65   123.8 3802.61   143.5 3789.52   149.6 3786.82   156.1 3785.11
   161.1 3784.16   195.2 3784.24     203 3784.96     210  3786.9   224.5 3791.16
   229.4 3791.55   247.2 3791.39   278.3 3792.74   307.3 3790.97   330.5 3791.38
   344.8 3790.63   355.9 3791.67   366.4 3791.66   382.2 3790.18   415.3 3793.23
     431 3793.63   444.7  3795.9   451.1 3795.75   465.4 3793.91   502.6 3795.07
#Mann= 7 ,-1,0
       0     .12       0      90      .1       0   156.1    .045       0
     203      .1       0     210     .12       0     330      .1       0
     500     .12       0
#XS Ineff= 2 , 0
                          266.39         3796.19
Permanent Ineff=
       F       F
Bank Sta=156.1,203
XS Rating Curve= 0 ,0
Exp/Cntr(USF)=0,0
Exp/Cntr=0.3,0.1

Type RM Length L Ch R = 1 ,23168   ,215.8,220.6,226
XS GIS Cut Line= 3
2266408.12574916541875.4743705422266661.53112281541510.331194341
2266741.34383891541446.481021454
#Sta/Elev= 30
       0 3797.98    16.1 3796.76    28.1 3795.18    66.1 3791.47   114.8 3790.48
   153.7 3790.37     168 3787.62   192.63783.881     217 3783.44   234.5 3783.85
   266.7 3787.41   285.2 3789.89   290.1 3789.82   309.5 3787.07   333.9 3786.87
   343.6 3787.98   357.9 3787.25   369.6 3788.58   415.6    3789     421 3789.33
   432.8 3793.22   441.4 3794.64   447.8 3794.63   455.7 3793.41   461.4 3793.16
   481.3 3794.62   506.9 3795.69   515.5 3796.78   524.7 3796.77   546.7 3797.94
#Mann= 3 ,-1,0
       0     .12       0   192.6    .045       0   234.5     .12       0
#XS Ineff= 2 , 0
                          288.94         3791.84
Permanent Ineff=
       F       F
Bank Sta=192.6,234.5
XS Rating Curve= 0 ,0
Exp/Cntr(USF)=0,0
Exp/Cntr=0.3,0.1

Type RM Length L Ch R = 1 ,22947   ,182.1,209,241.2
XS GIS Cut Line= 4
 2266438.0555177541979.2309014842266629.60603636541915.380728596
2266791.22678648 541735.802117352266896.97863533 541691.90512349
#Sta/Elev= 30
       0 3796.41    40.2 3792.03    65.5 3790.61      95 3790.78   116.1 3788.94
   145.6 3788.94     192 3790.64     211 3790.14   231.8 3788.21   247.6 3788.33
   284.6 3783.08   293.1 3782.38   344.1 3782.55   349.4 3783.12   369.6 3786.73
   412.1 3787.55   414.9 3787.97     421 3790.52   438.9 3792.86   444.5 3792.86
   457.5 3790.23   466.2 3789.79   487.8 3790.36   496.5 3792.52   505.2 3792.57
   509.5 3793.94   526.8 3804.36   531.2 3806.18   539.8 3808.14     558    3810
#Mann= 5 ,-1,0
       0      .1       0      50     .12       0     120      .1       0
   284.6    .045       0   349.4      .1       0
#XS Ineff= 2 , 0
          193.74 3792.19   440.5         3793.55
Permanent Ineff=
       F       F
Bank Sta=284.6,349.4
XS Rating Curve= 0 ,0
Exp/Cntr(USF)=0,0
Exp/Cntr=0.3,0.1

Type RM Length L Ch R = 1 ,22738   ,217.9,231.1,246.1
XS GIS Cut Line= 2
2266432.06956399542017.1419416362266916.93181436542009.160670025
#Sta/Elev= 30
       0 3796.77    32.1  3794.3    48.1 3794.64    72.1 3790.26    88.1 3790.38
   100.1 3789.58   108.1 3788.31   124.1 3787.72   156.1  3789.4   188.1 3789.02
   204.1 3789.48   272.1 3785.95   284.1 3786.74   292.1 3786.33   308.1 3786.91
   324.1 3788.06   332.2 3786.96   349.9 3782.29   352.2 3781.67   372.2 3781.53
   389.7 3781.64   393.6 3782.28   400.2 3785.49   404.2 3788.65   412.2 3791.35
   428.2 3790.76   436.2 3794.85   451.6 3806.14   460.2 3810.91   484.9 3814.96
#Mann= 4 ,-1,0
       0      .1       0      60     .12       0   349.9    .045       0
   393.6     .12       0
#XS Ineff= 2 , 0
          197.98 3791.05
Permanent Ineff=
       F       F
Bank Sta=349.9,393.6
XS Rating Curve= 0 ,0
Exp/Cntr(USF)=0,0
Exp/Cntr=0.3,0.1

Type RM Length L Ch R = 1 ,22507   ,243.8,241.1,240.6
XS GIS Cut Line= 4
 2266440.0508356542142.8469695082266527.84482332  542136.8610158
2266841.10973405542272.542633186 2266946.8615829542256.580089964
#Sta/Elev= 30
       0 3796.19    16.2 3794.48    28.2 3794.15      50 3790.98    60.3 3789.93
    91.5 3790.25   140.7  3785.7   162.5 3786.23   179.9  3788.5   197.3 3788.56
   223.5 3787.05   259.9 3787.12   271.4 3788.05   275.8 3787.81   288.9 3784.82
     302 3783.44   310.2 3781.27   356.2 3780.92   360.5 3781.12   389.6 3788.23
   415.3 3789.55   444.6 3789.06   452.7 3790.84   464.8 3789.27   468.9 3789.98
   481.4 3796.22   489.1  3799.2   505.3 3803.78   517.4 3805.67   536.3 3807.14
#Mann= 5 ,-1,0
       0      .1       0      50     .12       0   310.2    .045       0
   360.5     .12       0     368      .1       0
#XS Ineff= 2 , 0
          271.82 3790.24
Permanent Ineff=
       F       F
Bank Sta=310.2,360.5
XS Rating Curve= 0 ,0
Exp/Cntr(USF)=0,0
Exp/Cntr=0.3,0.1

Type RM Length L Ch R = 1 ,22266   ,268.3,240.1,212.7
XS GIS Cut Line= 3
2266402.13979545542354.350667198 2266807.1893297542509.985463611
2266960.82880822542428.177429599
#Sta/Elev= 30
       0 3806.48    25.4 3800.65    40.9 3798.73    96.5 3788.31   109.3 3785.06
   115.2 3785.21   146.2 3782.89   164.7 3783.87   186.3 3783.54   215.13780.581
   237.9 3779.67   266.9  3780.4   273.1  3780.6     285 3782.35   293.6  3781.3
   302.1 3782.78   327.8 3784.61   349.3 3783.67   379.3 3784.17   392.1 3783.08
     431 3786.94     450 3785.99   484.9 3785.74   521.1 3787.29   552.9 3786.75
   561.9 3788.59   566.5  3788.8   580.1 3787.18   593.6 3790.27     608 3790.55
#Mann= 4 ,-1,0
       0     .12       0   215.1    .045       0   266.9     .12       0
  523.92      .1       0
#XS Ineff= 2 , 0
                          429.65         3789.38
Permanent Ineff=
       F       F
Bank Sta=215.1,266.9
XS Rating Curve= 0 ,0
Exp/Cntr(USF)=0,0
Exp/Cntr=0.3,0.1

Type RM Length L Ch R = 1 ,22026   ,210.3,198.6,184.5
XS GIS Cut Line= 3
2266302.37390031542683.5781211492266565.75586347 542713.50788969
2266968.81007983542440.149337015
#Sta/Elev= 30
       0 3791.46      26 3792.22    71.8 3789.59    90.4 3791.16   158.8 3789.57
   174.9 3785.93   223.2 3786.68   243.4 3784.74   287.3 3784.18   314.4 3778.89
   340.5 3778.38   345.3 3778.84   359.8 3780.97   374.3 3780.63   393.8 3782.69
     413  3781.5   422.7 3783.26   439.9  3783.4     471 3782.08   485.5 3783.85
   506.1 3782.55   546.4 3784.56   557.9 3786.56   618.4 3785.39   683.7 3788.21
   698.2 3787.37   707.8 3788.72   722.3 3786.64   736.5 3789.67   752.1 3790.76
#Mann= 7 ,-1,0
       0      .1       0     190     .12       0   314.4    .045       0
   345.3     .12       0  415.08      .1       0  595.08     .12       0
  645.08      .1       0
#XS Ineff= 2 , 0
          224.36 3787.67  558.39          3787.6
Permanent Ineff=
       F       F
Bank Sta=314.4,345.3
XS Rating Curve= 0 ,0
Exp/Cntr(USF)=0,0
Exp/Cntr=0.3,0.1

Type RM Length L Ch R = 1 ,21827   ,202.4,194.2,187.2
XS GIS Cut Line= 3
2266699.44216296542942.969448504 2266883.6898181542584.829838143
2267006.24224368542490.690739492
#Sta/Elev= 30
       0 3817.38    64.2 3810.94      74  3811.3      94 3809.73    97.8 3808.46
   102.9 3805.42     119 3797.58   141.5 3782.95     146 3780.82   159.43778.185
     164 3777.67   197.9 3778.15   228.9 3780.79   240.4 3780.21   253.9 3782.41
   266.2 3782.17   278.1 3783.47   319.7  3782.5   339.4  3786.3   343.9 3786.41
   370.9  3783.8   402.4 3785.97     420 3784.63     474  3785.4   484.1 3786.73
     497 3786.68   505.5 3787.97   519.4 3786.07   536.9 3788.04   557.3 3788.37
#Mann= 6 ,-1,0
       0      .1       0     130     .12       0   159.4    .045       0
   197.9      .1       0     240     .12       0     360      .1       0
#XS Ineff= 2 , 0
                          343.63         3787.75
Permanent Ineff=
       F       F
Bank Sta=159.4,197.9
XS Rating Curve= 0 ,0
Exp/Cntr(USF)=0,0
Exp/Cntr=0.3,0.1

Type RM Length L Ch R = 1 ,21633   ,166.3,179.1,191.8
XS GIS Cut Line= 3
2266914.39416905543043.2722836892267006.51799662 542673.16076591
 2267114.8038992542574.572108336
#Sta/Elev= 30
       0 3846.48    47.5 3832.21    76.4 3821.12    88.7 3817.78   109.3 3809.59
   117.6 3807.24   126.7 3801.52   142.3 3789.24   158.3 3779.65   162.9 3777.26
   164.9 3776.85   204.1    3776   214.5 3776.49   241.2 3778.88   253.6 3779.03
   270.1 3781.55   282.5 3781.56   303.1 3780.46   331.9  3782.8     369 3782.76
   381.4 3783.84   393.3 3783.32   411.1 3784.34   432.3 3784.28   444.9 3786.29
   456.2 3784.95     476  3784.2   506.2 3784.35     518 3785.52   527.8 3787.51
#Mann= 7 ,-1,0
       0      .1       0      20     .12       0     130      .1       0
   164.9    .045       0   214.5      .1       0     270     .12       0
     330      .1       0
#XS Ineff= 2 , 0
                          318.58         3786.31
Permanent Ineff=
       F       F
Bank Sta=164.9,214.5
XS Rating Curve= 0 ,0
Exp/Cntr(USF)=0,0
Exp/Cntr=0.3,0.1

Type RM Length L Ch R = 1 ,21454   ,130.4,129.5,128.5
XS GIS Cut Line= 4
2266943.70097893543068.7764391112267075.60365316542980.239027638
2267212.02354226542787.8056741322267320.43669917542696.557933737
#Sta/Elev= 30
       0 3847.32    19.8 3839.32    29.5 3837.07    49.1 3829.82      68 3821.94
   106.7 3807.93   159.8 3781.94   175.8 3780.22   184.4  3778.5   196.9 3779.14
   221.5 3778.65   236.1 3776.31   249.8 3775.43   277.4 3775.54   284.8 3776.25
   293.4 3779.67   299.2 3780.75   314.6 3781.38   345.1 3778.25   353.8 3779.39
   373.8 3779.85   382.4 3782.64   396.7 3784.85   419.4 3782.41   439.3 3781.36
   457.7  3782.2   499.5 3782.73   504.6 3783.49   510.3 3785.82   536.4 3799.32
#Mann= 5 ,-1,0
       0      .1       0  168.86     .12       0  228.86      .1       0
   236.1    .045       0   284.8      .1       0
#XS Ineff= 2 , 0
                          397.49         3787.52
Permanent Ineff=
       F       F
Bank Sta=236.1,284.8
XS Rating Curve= 0 ,0
Exp/Cntr(USF)=0,0
Exp/Cntr=0.3,0.1

Type RM Length L Ch R = 1 ,21324   ,152.2,165.7,181.4
XS GIS Cut Line= 5
  2266976.224926543149.182863815  2267116.258587543091.362513466
2267192.14779683543043.4800358332267298.75406779542884.474072372
2267404.45689577542817.619292281
#Sta/Elev= 30
       0 3853.86    17.3 3847.59    25.9 3841.94    47.5 3830.53    69.2 3823.63
   125.4 3798.51     150 3785.55   161.7 3781.66   175.1 3780.04     194 3781.71
   212.9 3779.42   245.8 3780.94   263.1  3778.1   268.1  3776.2   271.7 3776.31
   284.4  3778.2     3093775.405   335.2 3774.47   358.2 3775.62   369.2    3779
   392.1 3779.83   398.6 3779.88   412.6 3782.89     428 3784.51   447.7 3783.22
   456.4 3781.03   511.5 3784.68   523.1 3786.75   543.2 3791.78   557.7 3796.74
#Mann= 7 ,-1,0
       0      .1       0   271.7     .12       0     309    .045       0
   358.2     .12       0   392.1      .1       0   523.1     .12       0
   543.2      .1       0
#XS Ineff= 2 , 0
                          429.65         3787.49
Permanent Ineff=
       F       F
Bank Sta=309,358.2
XS Rating Curve= 0 ,0
Exp/Cntr(USF)=0,0
Exp/Cntr=0.3,0.1

Type RM Length L Ch R = 1 ,21159   ,200.2,216.9,233
XS GIS Cut Line= 4
2266971.70771113543161.8310654542267268.03700667543141.955320022
2267389.09836521543068.7764391112267494.80119319543044.383478807
#Sta/Elev= 30
       0 3856.51    20.5 3850.05    40.6 3839.42    64.6 3828.54    72.6 3823.93
    84.7 3819.07   100.7 3811.17   116.7 3805.05   160.8 3781.85   164.8 3780.54
   176.9 3779.46   188.9 3780.19   200.9 3777.96     217 3777.49   311.2 3780.13
   321.7 3777.27   343.9 3777.91   373.4 3774.42     386 3773.24     400 3773.29
   417.1 3774.61   423.4 3777.31   429.9 3781.61   436.9 3784.15   441.6 3784.38
   449.8 3782.21     458 3783.11   487.4 3793.49   499.1 3798.91   546.9 3808.05
#Mann= 5 ,-1,0
       0      .1       0   373.4    .045       0   417.1      .1       0
     427     .12       0  528.46      .1       0
Bank Sta=373.4,417.1
XS Rating Curve= 0 ,0
Exp/Cntr(USF)=0,0
Exp/Cntr=0.3,0.1

Type RM Length L Ch R = 1 ,20942   ,254.9,256.6,258.7
XS GIS Cut Line= 3
2267059.34167962543314.5129280952267446.91871556543302.768169431
2267578.82138979543259.402906669
#Sta/Elev= 30
       0 3829.23    20.8 3819.94    36.9 3811.24    48.9 3806.87    56.9 3802.59
    72.9 3795.37    80.9 3792.87    92.9 3785.32   112.9  3776.3   140.9 3774.67
   168.7 3777.45   208.9 3777.73   224.9 3777.32     257 3778.33     269  3777.6
     289 3772.94     321 3772.28     341 3772.96     349 3775.64     357 3779.99
     361 3781.31     365 3781.97     375 3781.61     385 3783.44   397.5 3783.16
   418.5 3791.87   422.8 3792.89   469.1 3799.38   515.4 3808.54   526.6 3811.49
#Mann= 4 ,-1,0
       0      .1       0     289    .045       0     341     .12       0
  417.75      .1       0
Bank Sta=289,341
XS Rating Curve= 0 ,0
Exp/Cntr(USF)=0,0
Exp/Cntr=0.3,0.1

Type RM Length L Ch R = 1 ,20685   ,221.9,222,222
XS GIS Cut Line= 3
 2267109.5739198543555.4102645272267499.07992759543563.491302033
 2267641.3061877543510.156454493
#Sta/Elev= 30
       0 3814.61    18.6 3807.89    30.6 3801.98    50.6 3793.83    66.6 3789.79
    82.6 3780.48    86.6 3778.75    94.6 3776.77   178.6 3775.47   194.6 3776.42
   222.6 3776.85   246.7 3774.85   254.7 3772.13   270.7 3771.31   298.2 3771.13
   307.1 3771.83   333.5 3774.46   342.7 3774.79   349.2 3775.86   366.7 3780.04
   378.7 3780.28   386.7 3781.88   399.3 3781.26   403.6 3783.16   407.8 3786.34
   416.4 3790.03   497.6 3800.92   518.9 3805.84   531.7 3809.96   541.5 3812.06
#Mann= 4 ,-1,0
       0      .1       0     170     .12       0   254.7    .045       0
   307.1      .1       0
Bank Sta=254.7,307.1
XS Rating Curve= 0 ,0
Exp/Cntr(USF)=0,0
Exp/Cntr=0.3,0.1

Type RM Length L Ch R = 1 ,20463   ,245.1,225.6,200.2
XS GIS Cut Line= 4
2267161.43073571543877.3579010272267291.52652399543780.689502786
2267556.23531544543787.0136036062267678.20011696543751.779327612
#Sta/Elev= 30
       0 3813.52    13.4 3810.29    33.8 3804.31    56.4 3799.44    67.8 3796.39
    94.2  3792.2     143 3786.14   153.6  3783.9   182.7 3775.56   194.7 3773.96
   214.7 3772.72   222.7 3772.87   237.4  3770.8   250.8 3770.04   278.8 3770.12
   284.83770.772   294.8 3772.47   302.8 3772.67   314.8 3774.57   330.8 3774.44
   342.8  3773.5   398.8 3774.55   406.8  3777.5   422.8 3780.17   435.1 3780.39
   447.5 3784.71   472.6 3789.55   501.7 3797.22   522.6 3800.74   553.8 3807.88
#Mann= 3 ,-1,0
       0      .1       0   237.4    .045       0   284.8      .1       0
Bank Sta=237.4,284.8
XS Rating Curve= 0 ,0
Exp/Cntr(USF)=0,0
Exp/Cntr=0.3,0.1

Type RM Length L Ch R = 1 ,20238   ,185.4,191.9,202.4
XS GIS Cut Line= 4
2267294.81579783544013.9410580532267437.04205794544017.173473056
2267577.65211055543908.8875704742267703.71629564543874.947212949
#Sta/Elev= 30
       0 3796.79    17.4 3793.08    25.4 3790.71    41.4 3787.05    57.4 3783.86
    65.4 3782.99   106.2 3780.46   129.4 3779.95   150.2 3777.66   166.4 3771.84
   178.7 3769.82   187.3 3768.76   211.9 3768.69   221.5 3769.69   227.2 3770.93
   258.6 3773.27   267.4 3773.21   282.5 3771.81   302.7 3772.34   315.6 3776.78
   326.5 3779.71   331.3 3780.04   338.9 3779.06   343.1 3779.52   351.3 3781.27
   367.2 3786.49   396.6 3794.17   421.8 3800.07   432.5 3803.18   450.3 3807.56
#Mann= 3 ,-1,0
       0      .1       0   178.7    .045       0   221.5      .1       0
Bank Sta=178.7,221.5
XS Rating Curve= 0 ,0
Exp/Cntr(USF)=0,0
Exp/Cntr=0.3,0.1

Type RM Length L Ch R = 1 ,20046   ,363.5,389.9,413.3
XS GIS Cut Line= 3
2267322.24358512544170.9768676442267498.41496509544184.528512257
2267745.95834002544077.922241301
#Sta/Elev= 30
       0 3797.69      22 3793.68    46.1 3787.22    62.1 3783.81    86.2 3780.27
   110.3  3775.6   134.3 3774.12   166.4  3773.3   178.6 3773.78   198.8 3771.79
     211  3772.8   222.2 3772.45   238.4 3768.59   252.6 3767.31   265.7 3767.19
   293.2 3768.51   305.4 3771.28   309.3 3772.75   316.6 3776.45   326.6 3778.68
   335.4 3778.92   339.7    3778   344.1 3778.71   348.5 3780.78   357.1 3785.77
   378.9 3792.71     392 3796.22   400.7 3797.29   413.8 3801.46   446.2  3807.5
#Mann= 3 ,-1,0
       0      .1       0   238.4    .045       0   293.2      .1       0
Bank Sta=238.4,293.2
XS Rating Curve= 0 ,0
Exp/Cntr(USF)=0,0
Exp/Cntr=0.3,0.1

Type RM Length L Ch R = 1 ,19656   ,283.9,275,266.3
XS GIS Cut Line= 4
2267338.67385476544489.797202534 2267536.1185815544494.216964544
2267685.54608555544554.2245641612267811.61027064544525.132829139
#Sta/Elev= 30
       0  3800.5     5.5 3798.72    13.5 3795.04    21.5 3793.73    32.2 3790.54
    45.5 3785.15    55.7 3782.72    81.5  3772.8    85.5 3771.79   105.5 3770.18
   125.5 3769.95   169.5 3771.87     209 3771.54   253.6 3769.16   257.9 3768.63
   264.4  3766.4   271.5 3765.87   280.6 3765.13   296.7    3765   307.5 3765.82
   307.5 3765.83   322.6 3767.45   335.1 3773.02   339.8 3774.08   360.6 3776.18
   373.5 3774.28   385.8 3777.35   414.6 3781.53   443.3 3786.75   487.9 3793.02
#Mann= 3 ,-1,0
       0      .1       0   271.5    .045       0   307.5      .1       0
Bank Sta=271.5,307.5
XS Rating Curve= 0 ,0
Exp/Cntr(USF)=0,0
Exp/Cntr=0.3,0.1

Type RM Length L Ch R = 1 ,19381   ,301.2,294.4,287.9
XS GIS Cut Line= 2
2267342.68915687544753.2198199742267769.36793719 544814.63570502
#Sta/Elev= 30
       0 3800.29     9.6 3800.08    21.7  3797.3    37.9 3794.77    50.7 3792.12
    62.1  3790.8    82.3 3786.69    86.4 3785.51   102.5 3777.77   130.8 3767.65
   138.23764.456   155.1 3763.75   188.5 3764.26   195.5  3764.8   211.6 3767.77
   223.7 3769.15   264.2 3769.67   304.6 3773.39   316.7 3772.88   324.8 3774.16
   329.8 3773.93   336.9 3772.56     341 3772.67     345  3774.7     349 3777.49
   353.1  3778.8   381.4 3781.43   393.5 3781.98   409.7 3781.51   431.1 3783.68
#Mann= 3 ,-1,0
       0      .1       0   138.2    .045       0   188.5      .1       0
Bank Sta=138.2,188.5
XS Rating Curve= 0 ,0
Exp/Cntr(USF)=0,0
Exp/Cntr=0.3,0.1

Type RM Length L Ch R = 1 ,19086   ,242.6,239.5,238.2
XS GIS Cut Line= 3
2267371.78089189545076.461320217 2267646.5361671545061.915452706
2267772.60035219545078.077527718
#Sta/Elev= 30
       0 3804.81    16.4 3799.08    24.4 3796.86    39.2  3793.4    48.5 3791.88
    64.5 3786.29    79.6  3781.8   100.5 3770.28   108.5 3767.31   112.6 3766.88
   116.6 3765.68   121.4 3763.26   132.6 3762.37   168.6 3762.42   180.83762.952
   204.7 3766.82   224.7 3768.16   236.7 3767.01   244.7 3765.64   248.7 3765.58
   252.7 3766.45   260.8 3769.74   268.8 3771.95   276.8 3771.86   284.9 3769.95
   290.2 3769.65   321.2 3769.82   365.5 3773.22   393.9  3776.2   402.2 3777.77
#Mann= 3 ,-1,0
       0      .1       0   121.4    .045       0   180.8      .1       0
#XS Ineff= 2 , 0
                           271.4         3773.22
Permanent Ineff=
       F       F
Bank Sta=121.4,180.8
XS Rating Curve= 0 ,0
Exp/Cntr(USF)=0,0
Exp/Cntr=0.3,0.1

Type RM Length L Ch R = 1 ,18847   ,226.4,238.5,253.6
XS GIS Cut Line= 3
2267325.31522085545327.392151869 2267618.4322747545300.288862643
2267756.96019742545314.342420019
#Sta/Elev= 30
       0  3792.1      23  3786.1      31 3783.06    47.1 3779.88    75.2 3769.93
    79.2 3769.06    99.3  3766.9   131.4 3765.93   147.5  3766.9   192.2 3767.23
   195.9 3766.83   203.7 3763.55   206.9 3762.71   215.8 3761.11   231.8 3760.23
   255.9 3761.08     268  3763.9     280 3765.22   292.1 3769.81   296.1 3770.64
   300.1 3770.79   312.2 3768.99   320.2 3769.67   328.3 3769.62   340.3 3771.38
   352.4 3776.28   388.6 3785.29   400.7 3789.35   428.8 3797.21   433.6 3797.85
#Mann= 3 ,-1,0
       0      .1       0   215.8    .045       0   255.9      .1       0
Bank Sta=215.8,255.9
XS Rating Curve= 0 ,0
Exp/Cntr(USF)=0,0
Exp/Cntr=0.3,0.1

Type RM Length L Ch R = 1 ,18608   ,349.8,347,342.9
XS GIS Cut Line= 4
2267305.22580737545486.7258590712267493.95790937545524.141955141
2267602.37106627545561.2834996362267694.73181516545567.536234132
#Sta/Elev= 30
       0  3776.6    11.2 3773.42    27.5 3770.95    51.9 3769.58    80.5 3769.16
    93.1 3768.32   125.3 3764.82   133.5 3763.46   145.7 3763.31   150.9  3764.4
   161.1 3765.31   195.6 3766.05   207.4 3764.29   211.7 3764.17   228.6 3760.68
   245.4 3759.47   270.9 3759.91   275.1 3760.46     282 3763.67   287.8 3767.97
   289.4 3768.58   300.5 3770.84   304.7 3771.09   312.8 3770.37   317.7 3771.92
   336.9 3783.02   360.9 3789.74   368.7 3791.38     377 3794.08   399.6 3798.66
#Mann= 4 ,-1,0
       0      .1       0     170     .12       0   228.6    .045       0
   275.1      .1       0
Bank Sta=228.6,275.1
XS Rating Curve= 0 ,0
Exp/Cntr(USF)=0,0
Exp/Cntr=0.3,0.1

Type RM Length L Ch R = 1 ,18261   ,440.6,402.8,346.3
XS GIS Cut Line= 3
2267310.36500684545840.9274682912267568.95820704545902.343353338
2267704.71963714545803.754695763
#Sta/Elev= 30
       0 3778.47    38.9 3772.17    48.2 3771.55    67.6  3769.3    81.4 3766.18
    92.3 3765.19   112.9 3761.51   121.1  3759.1   125.2 3758.62   137.5 3758.59
   174.6 3758.59   184.4 3759.04   197.7 3761.41   223.9 3763.91   248.5 3763.83
   260.8 3765.78   279.6 3765.12   299.4 3765.58     309 3765.16   314.3 3765.68
   319.2 3767.04   322.2 3767.38   334.8 3764.95   343.9 3765.73   383.5 3766.69
   393.3 3768.96   397.1 3769.07   409.2 3766.73   413.1 3766.98   433.6 3770.32
#Mann= 5 ,-1,0
       0     .12       0   121.1    .045       0   184.4      .1       0
  265.79     .12       0  305.79      .1       0
#XS Ineff= 2 , 0
                          261.31          3768.1
Permanent Ineff=
       F       F
Bank Sta=121.1,184.4
XS Rating Curve= 0 ,0
Exp/Cntr(USF)=0,0
Exp/Cntr=0.3,0.1

Type RM Length L Ch R = 1 ,17859   ,401.8,372.7,339.2
XS GIS Cut Line= 2
2267484.91541697546343.5680011692267801.69208721545897.494730834
#Sta/Elev= 30
       0 3837.88    21.3 3825.06    33.3  3816.6      50 3803.65    72.9 3782.23
    84.4 3769.72    91.2 3761.17    96.1 3756.85   101.1 3755.97   115.9 3755.91
   153.2  3756.8   164.7 3759.24   178.3 3760.14   187.7 3759.77     202 3762.32
   218.8 3763.86   243.3 3763.69     258 3762.46   309.6 3763.11   356.2  3762.2
   419.9 3763.59   478.8 3765.91     486 3766.74   494.6 3766.04   503.3 3767.53
     509 3767.54   517.6 3766.38   527.9 3770.88   537.7 3769.62   547.1 3770.18
#Mann= 5 ,-1,0
       0      .1       0    96.1    .045       0   153.2     .12       0
     450      .1       0     490     .12       0
#XS Ineff= 2 , 0
                          218.79          3768.7
Permanent Ineff=
       F       F
Bank Sta=96.1,153.2
XS Rating Curve= 0 ,0
Exp/Cntr(USF)=0,0
Exp/Cntr=0.3,0.1

Type RM Length L Ch R = 1 ,17486   ,237,233.8,232.4
XS GIS Cut Line= 3
2267939.06972482546361.3462836832267846.94589725545983.153728398
2267876.03763227 545931.43508836
#Sta/Elev= 30
       0 3780.16    20.8 3775.86    37.2 3773.51      46 3769.44    57.8 3763.17
    61.9 3761.49    70.2    3760    86.6 3755.78    98.5 3754.15   110.6 3753.75
     136 3753.76   140.1  3754.2   148.4 3757.36   152.5 3758.14   164.9 3757.97
   173.1 3757.23   189.6 3757.22   197.8 3759.34     206 3760.01   308.9 3760.34
   337.8  3761.3   370.7 3764.53   391.5 3765.47   400.4 3767.04   405.3 3766.85
   409.9 3765.97   414.5 3766.05   426.9 3767.81     442 3770.72   448.6  3771.3
#Mann= 6 ,-1,0
       0      .1       0    98.5    .045       0   140.1     .12       0
     200      .1       0     300     .12       0  429.25      .1       0
#XS Ineff= 2 , 0
                          202.51         3762.74
Permanent Ineff=
       F       F
Bank Sta=98.5,140.1
XS Rating Curve= 0 ,0
Exp/Cntr(USF)=0,0
Exp/Cntr=0.3,0.1

Type RM Length L Ch R = 1 ,17252   ,252,254.1,257.4
XS GIS Cut Line= 3
2268176.65222749546301.5466061382268078.06356992546007.396840917
2268071.59873992 545918.50542835
#Sta/Elev= 30
       0 3773.93    21.5 3769.02    55.2 3758.57    63.7 3756.64    72.1 3756.36
    84.8  3757.5    93.2 3756.85   110.1 3756.77   125.13753.588   139.4  3753.1
   175.43753.403   190.2 3756.63   194.4 3756.87   221.8  3756.1   236.6 3754.52
   240.9 3754.73   253.2 3757.27   257.7 3757.57     283  3757.1   291.5 3758.78
   299.9 3763.12   308.4 3764.85   312.5 3765.08   324.5 3763.26   332.5 3759.92
   340.5 3759.62   362.7 3764.05   376.6 3770.14   384.6 3772.27   399.4 3774.93
#Mann= 4 ,-1,0
       0      .1       0      40     .12       0   125.1    .045       0
   175.4      .1       0
#XS Ineff= 2 , 0
                          264.16         3766.88
Permanent Ineff=
       F       F
Bank Sta=125.1,175.4
XS Rating Curve= 0 ,0
Exp/Cntr(USF)=0,0
Exp/Cntr=0.3,0.1

Type RM Length L Ch R = 1 ,16998   ,140.1,151.9,167
XS GIS Cut Line= 3
2268419.98631162546279.7530215172268352.10559657546003.381538809
2268337.55972906545866.003901206
#Sta/Elev= 30
       0 3773.75      45 3763.21    61.5 3760.51      78 3758.92    97.9 3758.36
     118 3755.79   150.9 3755.68   159.2  3754.2   179.8 3752.76   208.6 3751.77
   225.1 3752.67   233.3 3753.12   237.4 3753.89   241.5 3755.41     258 3754.43
   262.1 3755.46   270.4 3760.77   274.5 3762.39   282.7 3763.46   294.8 3762.23
   298.9 3760.91   306.9 3756.88   310.9 3756.21   351.2  3756.2   367.2 3756.97
   375.3 3758.59   383.3  3761.2   395.4 3762.44   407.5 3768.06   422.7 3771.62
#Mann= 5 ,-1,0
       0      .1       0      10     .12       0     110      .1       0
   179.8    .045       0   225.1      .1       0
#XS Ineff= 2 , 0
                          281.84         3764.05
Permanent Ineff=
       F       F
Bank Sta=179.8,225.1
XS Rating Curve= 0 ,0
Exp/Cntr(USF)=0,0
Exp/Cntr=0.3,0.1

Type RM Length L Ch R = 1 ,16846   ,178.4,197.2,215.3
XS GIS Cut Line= 3
2268490.19648273546306.3952286412268535.45029276546009.013048418
2268575.85548029545861.938165807
#Sta/Elev= 30
       0 3776.12    17.4 3771.67    90.6    3758   126.7 3754.81   138.8 3754.68
   171.2 3756.08   179.3 3754.88   191.4 3754.58   199.5 3751.91   199.5  3751.9
   223.8 3751.07   248.6 3751.17     2553751.741   260.2 3752.66   268.3 3752.69
   272.3 3753.48   284.5 3759.81   292.5 3761.94   296.6 3762.38   301.3 3762.06
   321.4 3755.62   375.3 3755.09   379.4 3755.71   395.6 3758.52   408.6 3761.98
   420.9 3763.21   425.1 3766.25   429.2 3770.28   433.4 3773.14   453.3 3783.07
#Mann= 5 ,-1,0
       0     .12       0      40      .1       0     140     .12       0
   199.5    .045       0     255      .1       0
#XS Ineff= 2 , 0
                          296.45         3763.01
Permanent Ineff=
       F       F
Bank Sta=199.5,255
XS Rating Curve= 0 ,0
Exp/Cntr(USF)=0,0
Exp/Cntr=0.3,0.1

Type RM Length L Ch R = 1 ,16649   ,165.4,181.3,201.4
XS GIS Cut Line= 2
2268530.67130881546339.2308940582268807.04279152 546009.52456381
#Sta/Elev= 30
       0 3777.32    13.9 3774.62    28.8    3773    45.9 3768.58      65 3764.45
    89.5 3757.27   107.1 3754.62   117.5 3754.06   130.3 3754.59   138.4 3753.34
   147.3 3752.92   159.3 3754.26     207 3755.41   221.9 3753.42     239 3754.06
   256.73751.515   263.6 3750.38   268.9 3750.27   300.2 3750.43   303.5 3751.46
   306.3    3753   315.8 3760.35   320.5 3762.17   326.2 3762.65   337.6 3760.87
   343.2 3761.01   351.8 3762.12   378.5 3777.05   411.4 3786.81   430.2 3792.98
#Mann= 4 ,-1,0
       0     .12       0     220      .1       0   256.7    .045       0
   303.5      .1       0
Bank Sta=256.7,303.5
XS Rating Curve= 0 ,0
Exp/Cntr(USF)=0,0
Exp/Cntr=0.3,0.1

Type RM Length L Ch R = 1 ,16468   ,288.5,285.4,282
XS GIS Cut Line= 4
2268627.57412033546409.8325087192268732.62760791 546304.77902114
2268876.47007552546241.7469285932268950.81562058546170.633798539
#Sta/Elev= 30
       0 3769.36     9.4 3766.79    23.6 3761.83      49 3755.96    54.6 3755.13
    63.1 3754.97    74.4 3753.88   108.4 3752.94     131 3755.28     148 3756.16
   167.5 3753.46   200.5 3752.62   205.6 3752.23   213.6 3750.69   222.3 3749.92
   281.5 3750.62   283.5 3750.82   292.2 3757.23   296.7  3759.7   300.9 3761.09
   308.6 3762.24     318 3761.44   321.8 3761.72   328.4 3766.26   334.1 3768.67
   349.5 3772.02   365.2 3776.92   381.7 3780.38     399 3786.23   408.5 3788.53
#Mann= 5 ,-1,0
       0     .12       0  168.57      .1       0   213.6    .045       0
   281.5      .1       0  405.61     .12       0
Bank Sta=213.6,281.5
XS Rating Curve= 0 ,0
Exp/Cntr(USF)=0,0
Exp/Cntr=0.3,0.1

Type RM Length L Ch R = 1 ,16182   ,403.8,381.2,356.1
XS GIS Cut Line= 2
2268755.25451293546626.4043138822269049.40427815546388.821811203
#Sta/Elev= 30
       0 3787.04    15.7 3782.04      32  3777.7    42.3 3775.76    52.9 3772.71
    62.9 3769.09      68 3766.58    89.7 3754.09    93.7 3752.62   101.1 3751.59
   110.83748.974   122.9 3748.15   150.3 3748.72   165.7 3750.42     176 3750.18
   199.3 3751.38   217.1 3751.18   257.5 3754.77   269.3 3754.72   275.7 3755.39
   288.4 3758.82   294.8 3759.91   314.8 3761.12   325.1 3760.28   337.2 3762.44
   352.1 3761.07   361.1 3762.54   364.8 3763.67   368.5 3765.58   378.1 3768.21
#Mann= 5 ,-1,0
       0      .1       0   110.8    .045       0   150.3      .1       0
     250     .12       0  378.11      .1       0
Bank Sta=110.8,150.3
XS Rating Curve= 0 ,0
Exp/Cntr(USF)=0,0
Exp/Cntr=0.3,0.1

Type RM Length L Ch R = 1 ,15801   ,227.3,223.1,219.8
XS GIS Cut Line= 3
2269167.38742574546813.8843840232269199.71157576546519.734618802
2269225.57089578546471.248393765
#Sta/Elev= 30
       0 3779.24    32.9 3768.79      49 3762.15    54.2 3758.69    65.1 3749.21
    67.7 3747.76    69.1 3746.96    73.9 3746.68    97.3 3746.26   105.3  3746.4
   110.1 3747.33   121.4 3749.19   149.6  3750.4   161.7 3751.59   173.7 3750.04
   185.8 3751.11   201.9 3750.24     214 3750.86     222 3752.83   234.1 3753.15
   238.1 3753.98   242.2 3755.05   250.2 3759.21   258.3 3760.37   278.4 3759.83
   294.5 3761.26   307.9 3759.84   312.4 3761.92   321.5 3767.81   350.9 3771.05
#Mann= 4 ,-1,0
       0     .12       0    67.7    .045       0   110.1     .12       0
     250      .1       0
Bank Sta=67.7,110.1
XS Rating Curve= 0 ,0
Exp/Cntr(USF)=0,0
Exp/Cntr=0.3,0.1

Type RM Length L Ch R = 1 ,15578   ,225.8,241.9,256
XS GIS Cut Line= 3
2269401.73751342 546810.651969022269398.50509841546602.161201364
2269421.13200343546534.280486313
#Sta/Elev= 30
       0  3771.3    29.5 3762.06    45.5  3756.2    49.5 3754.45    53.5 3752.21
    61.5 3747.09    65.5 3746.01   109.6 3745.88   117.5 3746.22   121.8    3747
   125.5 3747.78   129.5 3748.02   133.5 3747.73   137.5 3748.04   145.5 3749.67
   161.5 3750.91   169.5 3752.68   185.5    3755   197.5 3757.32   213.8 3758.25
   222.2 3759.89   226.4    3760   234.8 3758.73   239.1 3759.25   243.3  3761.1
   247.5 3763.76   248.6    3764   251.7 3764.41   264.4 3764.44   280.1 3767.28
#Mann= 6 ,-1,0
       0     .12       0      50      .1       0    61.5    .045       0
   121.8      .1       0     150     .12       0  248.52      .1       0
Bank Sta=61.5,121.8
XS Rating Curve= 0 ,0
Exp/Cntr(USF)=0,0
Exp/Cntr=0.3,0.1

Type RM Length L Ch R = 1 ,15336   ,211.9,243.9,281.6
XS GIS Cut Line= 3
2269502.60039578546864.6208207822269597.96382084546823.463974179
2269683.28899063546639.763902757
#Sta/Elev= 30
       0 3767.82     6.9 3766.97    27.9 3762.76    40.9 3761.34    79.9 3753.22
    92.1 3752.26   106.4 3752.64   115.2  3751.9   134.4 3751.71   150.5  3748.5
   166.1 3746.39   175.6 3744.68   181.4 3744.06   191.6 3743.96   212.7 3744.13
   218.7  3744.7   221.1 3745.18   225.5 3747.39   234.3 3754.32   238.7 3756.33
   251.9 3758.69   256.3 3758.72   263.9 3757.91   266.9 3758.39   272.9 3761.61
   278.4 3765.15   282.8 3768.58   287.2 3771.21     296 3775.13   306.4 3778.07
#Mann= 4 ,-1,0
       0     .12       0  173.87      .1       0   175.6    .045       0
   218.7      .1       0
#XS Ineff= 2 , 0
          131.52  3753.6
Permanent Ineff=
       F       F
Bank Sta=175.6,218.7
XS Rating Curve= 0 ,0
Exp/Cntr(USF)=0,0
Exp/Cntr=0.3,0.1

Type RM Length L Ch R = 1 ,15092   ,124.9,130.9,142.1
XS GIS Cut Line= 2
2269598.91482856546944.7971916212269883.36734878546906.008211592
#Sta/Elev= 30
       0 3753.92    17.4 3751.77    33.6 3750.64    49.7 3750.72      58 3750.08
    73.9  3749.8    98.2 3750.44   110.3 3750.07   134.5 3750.16   146.6 3747.66
   157.1  3744.7   162.8 3743.46   166.8 3743.31   202.9 3743.12   210.4 3743.54
   213.33744.274   219.3 3746.84   223.3 3749.66   227.3 3752.94   231.4 3755.16
   235.4 3756.66   239.5 3757.23   243.5 3757.29   251.6  3756.7   255.6 3758.47
   259.6 3761.91   267.2 3771.46   279.8 3786.01   283.9  3789.9   287.1 3792.07
#Mann= 4 ,-1,0
       0     .12       0     140      .1       0   157.1    .045       0
   213.3      .1       0
#XS Ineff= 2 , 0
          124.22 3753.78
Permanent Ineff=
       F       F
Bank Sta=157.1,213.3
XS Rating Curve= 0 ,0
Exp/Cntr(USF)=0,0
Exp/Cntr=0.3,0.1

Type RM Length L Ch R = 1 ,14961   ,231.1,248.1,265.8
XS GIS Cut Line= 2
2269569.85670609547023.2252540322269903.12678102547068.397402743
#Sta/Elev= 30
       0 3753.18    10.4 3752.21    22.5 3751.85    62.9 3749.21    95.2 3749.75
   119.4 3749.23   131.5  3748.2   147.7 3748.23   163.8 3748.94   171.9 3748.22
     188 3743.79   199.3 3741.92   204.2 3741.41   224.4 3741.22   232.4 3741.87
   240.5 3742.35   244.5 3743.69   248.6 3745.79   256.6 3752.17   260.7 3754.56
   264.7 3755.68   276.8 3755.39   280.9 3756.88   284.9 3760.43   288.9 3766.18
     293 3771.27   309.5 3785.56   317.2 3790.86   329.3 3796.97   336.3 3799.68
#Mann= 6 ,-1,0
       0      .1       0      70     .12       0   199.3    .045       0
   232.4     .12       0     270      .1       0     280     .12       0
#XS Ineff= 2 , 0
           162.7 3750.88
Permanent Ineff=
       F       F
Bank Sta=199.3,232.4
XS Rating Curve= 0 ,0
Exp/Cntr(USF)=0,0
Exp/Cntr=0.3,0.1

Type RM Length L Ch R = 1 ,14713   ,267.8,271.1,271.1
XS GIS Cut Line= 3
  2269510.023416547140.3582992682269750.83833368547326.222161908
2269821.95146373547348.849066925
#Sta/Elev= 30
       0 3754.14    22.9 3752.18    63.4 3747.69    78.5 3747.11    99.1 3747.21
     129 3745.59   141.9 3746.72   174.5 3746.84   179.6 3746.24   190.3 3742.05
   194.7 3741.24   235.1  3740.4   250.3 3740.44   256.7 3741.01   260.4 3741.73
   261.6 3742.35   278.7 3752.61   281.6 3753.95   285.7 3754.64   295.8 3753.53
   309.8 3753.27     314 3754.46   318.2 3756.68   322.4 3762.91   330.8 3776.41
     335 3782.45   339.2 3786.13     349 3790.82   360.2 3794.75   378.8 3802.47
#Mann= 4 ,-1,0
       0      .1       0      40     .12       0   194.7    .045       0
   256.7     .12       0
#XS Ineff= 2 , 0
          146.14 3750.26
Permanent Ineff=
       F       F
Bank Sta=194.7,256.7
XS Rating Curve= 0 ,0
Exp/Cntr(USF)=0,0
Exp/Cntr=0.3,0.1

Type RM Length L Ch R = 1 ,14442   ,117.3,113.9,112
BEGIN DESCRIPTION:
Structure XS 4
END DESCRIPTION:
XS GIS Cut Line= 3
2269342.99213701547339.430295005 2269641.1283185547587.375200149
2269787.68684542 547606.44788516
#Sta/Elev= 30
       0 3753.99    32.8 3749.73    84.1 3745.78   149.8 3745.61   162.8 3742.84
   178.4 3742.22   190.4 3739.81   199.2 3738.94     235 3738.82   245.53739.611
   257.7 3743.05   277.6 3745.41   298.1 3745.35   314.5 3743.06   324.1 3744.17
   342.9 3745.03   355.3 3747.64   365.7 3746.81   374.2 3746.97   390.8 3753.06
   394.9 3753.39   402.9 3750.98     415 3751.42   423.1 3750.13   427.1 3752.05
   447.3 3769.68   451.3 3772.59   459.4 3776.53     517 3795.97   535.6 3800.99
#Mann= 5 ,-1,0
       0      .1       0      30     .12       0     180      .1       0
   190.4    .045       0   245.5      .1       0
#XS Ineff= 2 , 0
          146.97 3748.25  290.19         3748.25
Permanent Ineff=
       F       F
Bank Sta=190.4,245.5
XS Rating Curve= 0 ,0
Exp/Cntr(USF)=0,0
Exp/Cntr=0.5,0.3
